--- DRPLKCR.prj (project) ---

Proj Title=DRPLKCR
Current Plan=p01
Default Exp/Contr=0,0
English Units
Geom File=g01
Flow File=f01
Plan File=p01
BEGIN DESCRIPTION:
Stream Name: Dropping Lick Creek
Flood Zone: Approximate
Monroe County, West Virginia
HEC-RAS Version: 5.0.7
Vertical Datum: NAVD88
Projection: NAD 1983 StatePlane West Virginia S FIPS 4702 (US Feet)
LiDAR: 2016, 1-meter
Land Use: 2016 NLCD
Hydrology Method:
Regression.
Model Notes:
END DESCRIPTION:
DSS File=dss
DSS Export Rating Curves= 0
DSS Export Rating Curve Sorted= 0
DSS Export Volume Flow Curves= 0
DXF OffsetX= 0
DXF OffsetY= 0
DXF ScaleX= 0
DXF ScaleY= 0

--- DRPLKCR.p01 (plan) ---

Plan Title=Floodplain
Program Version=5.07
Short Identifier=Floodplain
Geom File=g01
Flow File=f01
Subcritical Flow
K Sum by GR= 0
Std Step Tol= 0.01
Critical Tol= 0.01
Num of Std Step Trials= 20
Max Error Tol= 0.3
Flow Tol Ratio= 0.001
Split Flow NTrial= 30
Split Flow Tol= 0.02
Split Flow Ratio= 0.02
Log Output Level= 0
Friction Slope Method= 1
Unsteady Friction Slope Method= 2
Unsteady Bridges Friction Slope Method= 1
Parabolic Critical Depth
Global Vel Dist= 0 , 0 , 0
Global Log Level= 0
CheckData=True
Encroach Param=-1 ,0,0, 0
Computation Interval=0.1SEC
Output Interval=1MIN
Instantaneous Interval=Max Profile
Mapping Interval=1HOUR
Computation Time Step Use Courant=        0
Computation Time Step Use Time Series=    0
Computation Time Step Count To Double=0
Computation Time Step Max Doubling=0
Computation Time Step Max Halving=0
Computation Time Step Residence Courant=0
Run HTab= 0
Run UNet= 0
Run Sediment= 0
Run PostProcess= 0
Run WQNet= 0
Run RASMapper=-1
UNET Theta= 0
UNET Theta Warmup= 0
UNET ZTol= 0
UNET ZSATol= 0
UNET MxIter= 0
UNET Max Iter WO Improvement= 0
UNET MaxInSteps= 0
UNET DtIC= 0
UNET DtMin= 0
UNET MaxCRTS= 0
UNET WFStab= 0
UNET SFStab= 0
UNET WFX= 1
UNET SFX= 1
UNET 1D Methodology=Finite Difference
UNET DSS MLevel= 1
UNET Pardiso=0
UNET DZMax Abort= 0
UNET Use Existing IB Tables= 0
UNET Froude Reduction=False
UNET Froude Limit= 0
UNET Froude Power= 0
UNET D1 Cores= 0
UNET D2 Coriolis=0
UNET D2 Cores= 0
UNET D2 Theta= 1
UNET D2 Theta Warmup= 1
UNET D2 Z Tol= 0.01
UNET D2 Volume Tol= 0.01
UNET D2 Max Iterations= 20
UNET D2 Equation= 0
UNET D2 RampUpFraction=0.1
UNET D2 TimeSlices= 1
UNET D2 BCVolumeCheck=0
UNET D1D2 MaxIter= 0
UNET D1D2 ZTol=0.01
UNET D1D2 QTol=0.1
UNET D1D2 MinQTol=1
DSS File=dss
Write IC File= 0
Write IC File at Fixed DateTime=0
Write IC File at Sim End=0
Echo Input=False
Echo Parameters=False
Echo Output=False
Write Detailed= 0
HDF Write Warmup=0
HDF Write Time Slices=0
HDF Flush=0
HDF Face Node Velocities=0
HDF Compression= 1
HDF Chunk Size= 1
HDF Spatial Parts= 1
HDF Use Max Rows=0
HDF Fixed Rows= 1
Calibration Method= 0
Calibration Iterations= 20
Calibration Max Change=0.05
Calibration Tolerance=0.2
Calibration Maximum=1.5
Calibration Minimum=0.5
Calibration Optimization Method= 1
WQ AD Non Conservative
WQ ULTIMATE=-1
WQ Max Comp Step=1HOUR
WQ Output Interval=15MIN
WQ Output Selected Increments= 0
WQ Output face flow=0
WQ Output face velocity=0
WQ Output face area=0
WQ Output face dispersion=0
WQ Output cell volume=0
WQ Output cell surface area=0
WQ Output cell continuity=0
WQ Output cumulative cell continuity=0
WQ Output face conc=0
WQ Output face dconc_dx=0
WQ Output face courant=0
WQ Output face peclet=0
WQ Output face adv mass=0
WQ Output face disp mass=0
WQ Output cell mass=0
WQ Output cell source sink temp=0
WQ Output nsm pathways=0
WQ Output nsm derived pathways=0
WQ Output MaxMinRange=-1
WQ Daily Max Min Mean=-1
WQ Daily Range=0
WQ Daily Time=0
WQ Create Restart=0
WQ Fixed Restart=0
WQ System Summary=0
WQ Write To DSS=0
WQ Use Fixed Temperature=0
Sorting and Armoring Iterations= 10
XS Update Threshold= 0.02
Bed Roughness Predictor= 0
Hydraulics Update Threshold= 0.02
Energy Slope Method= 1
Volume Change Method= 1
Sediment Retention Method= 0
XS Weighting Method= 0
Number of US Weighted Cross Sections= 1
Number of DS Weighted Cross Sections= 1
Upstream XS Weight=0
Main XS Weight=1
Downstream XS Weight=0
Number of DS XS's Weighted with US Boundary= 1
Upstream Boundary Weight= 1
Weight of XSs Associated with US Boundary= 0
Number of US XS's Weighted with DS Boundary= 1
Downstream Boundary Weight= 0.5
Weight of XSs Associated with DS Boundary= 0.5
Percentile Method= 0
Sediment Output Level= 3
Mass or Volume Output= 0
Output Increment Type= 1
Profile and TS Output Increment= 1
XS Output Flag= 0
XS Output Increment= 10
Write Gradation File= 0
Read Gradation Hotstart= 0
Write HDF5 File= 1
Write Binary Output= 1
Write DSS Sediment File= 0
SV Curve= 0
Specific Gage Flag= 0

--- DRPLKCR.f01 (steady flow) ---

Flow Title=Flow
Program Version=5.07
Number of Profiles= 6
Profile Names=01pct,10pct,04pct,02pct,0_2pct,01plus
River Rch & RM=DRPLKCR,Main            ,39084
     550     290     386     465     769     813
River Rch & RM=DRPLKCR,Main            ,37005
     573     303     402     485     800     847
River Rch & RM=DRPLKCR,Main            ,36412
     626     332     440     530     872     925
River Rch & RM=DRPLKCR,Main            ,33969
     692     368     488     587     963    1020
River Rch & RM=DRPLKCR,Main            ,31070
    1050     567     745     891    1450    1550
River Rch & RM=DRPLKCR,Main            ,28359
    1270     694     909    1090    1750    1880
River Rch & RM=DRPLKCR,Main            ,27956
    1350     738     966    1150    1860    2000
River Rch & RM=DRPLKCR,Main            ,23458
    1790     990    1290    1530    2450    2650
River Rch & RM=DRPLKCR,Main            ,19955
    1920    1060    1380    1640    2620    2830
River Rch & RM=DRPLKCR,Main            ,12951
    2130    1180    1530    1820    2900    3140
River Rch & RM=DRPLKCR,Main            ,8568
    2320    1300    1680    1990    3160    3440
River Rch & RM=DRPLKCR,Main            ,934
    2330    1300    1680    2000    3170    3440
River Rch & RM=DRPLKCR,Main            ,0
    3730    2120    2720    3210    5030    5510
Boundary for River Rch & Prof#=DRPLKCR,Main            , 1
Up Type= 0
Dn Type= 1
Dn Known WS=1807.751
Boundary for River Rch & Prof#=DRPLKCR,Main            , 2
Up Type= 0
Dn Type= 1
Dn Known WS=1806.125
Boundary for River Rch & Prof#=DRPLKCR,Main            , 3
Up Type= 0
Dn Type= 1
Dn Known WS=1807.067
Boundary for River Rch & Prof#=DRPLKCR,Main            , 4
Up Type= 0
Dn Type= 1
Dn Known WS=1807.447
Boundary for River Rch & Prof#=DRPLKCR,Main            , 5
Up Type= 0
Dn Type= 1
Dn Known WS=1808.816
Boundary for River Rch & Prof#=DRPLKCR,Main            , 6
Up Type= 0
Dn Type= 1
Dn Known WS=1809.173
DSS Import GetInterval= 0
DSS Import GetPeak= 0
DSS Import FillOption= 0

--- DRPLKCR.g01 (geometry) ---

Geom Title=Geometry
Program Version=5.07

River Reach=DRPLKCR         ,Main
Reach XY= 30
2112316.12009516185383.8888099872111495.23989873 184689.97201959
2110156.81200004185026.4910000062109312.02000003184798.886000005
2107711.11200004185122.7750000272106150.74600001183867.534999995
2105208.35600002183509.799000024     2104412.935183473.977000031
2104067.44900005183867.6399999912103406.85800004183914.949000015
     2103061.806183236.1300000352101422.04900002182792.987000017
2100252.77800005182850.2789999972099774.82700001183436.824000021
2098891.14700003183658.1780000082098724.48000004183019.289000041
2098148.34400005183423.7470000062097330.50600005182908.837000042
     2096702.584183412.4460000142096442.36200004184363.039000043
2095096.00799999186264.949000023     2093784.376185478.491000023
     2092549.133185471.5460000312091780.03600006184885.175000018
2090987.24000001 184888.647000032089376.12900004183113.473000011
     2087714.671181977.1889999952084729.52599999181572.206000022
     2083539.422 182158.144000022082090.73099516181876.368496227

Type RM Length L Ch R = 1 ,39084   ,97.1,100.3,99.9
XS GIS Cut Line= 4
2112523.23171169185306.4061300442112319.24296974185352.503581569
 2112298.5977548185429.3496593972112260.74819407185545.192254332
#Sta/Elev= 30
       02408.979   8.4912408.377  21.0152406.818   47.39 2404.33  60.8442403.731
  67.5712402.675  74.2982402.121 101.2072402.447 111.2982401.761 114.661 2401.79
 125.2712402.186 138.9882402.276 157.3342403.457 168.4782402.476 178.569 2402.13
 196.6032402.196 210.899 2401.91 227.8852402.195 231.2822401.811 234.6792400.904
 238.0762400.415 248.2682402.246 258.4592403.285 295.7742404.114 330.4572405.234
 358.0692406.984 375.3272411.357 386.8272414.756 402.4362418.289 410.5732419.769
#Mann= 5 ,-1 , 0
       0    .035       0     150     .04       0 227.885    .045       0
 248.268     .04       0   298.7      .1       0
#XS Ineff= 2 , 0
           153.3 2406.36
Permanent Ineff=
       F       F
Bank Sta=227.885,248.268
XS Rating Curve= 0 ,0
Exp/Cntr(USF)=0,0
Exp/Cntr=0.3,0.1

Type RM Length L Ch R = 1 ,38984   ,99.9,105.5,106.4
XS GIS Cut Line= 4
2112529.39341627185289.1571804022112240.10297914 185296.30271868
2112202.25341841    185413.292272112175.87342155185515.371388309
#Sta/Elev= 30
       02406.284  18.5612404.268  39.2752400.905  52.4022399.873 108.1932400.311
 121.321 2400.54 131.1662401.008 183.6752400.581  209.932400.078 232.9032400.333
 242.7452399.628 259.1582399.826  282.132398.771 305.4132399.195  312.312398.833
 319.2062399.188  324.32 2398.28 329.6092397.261 332.9992397.003 339.8962397.511
 343.3442398.292 350.2412400.106 364.0342400.658  370.93 2401.79 398.5162405.038
 408.8612406.578 425.8642408.659 446.1962411.617 494.355 2420.27 517.7712425.479
#Mann= 4 ,-1 , 0
       0    .035       0     150     .04       0  324.32    .045       0
 343.344      .1       0
#XS Ineff= 2 , 0
          258.74 2401.95
Permanent Ineff=
       F       F
Bank Sta=324.32,343.344
XS Rating Curve= 0 ,0
Exp/Cntr(USF)=0,0
Exp/Cntr=0.3,0.1

Type RM Length L Ch R = 1 ,38879   ,129.4,128.3,127.4
XS GIS Cut Line= 4
2112567.32326394185253.9316010122112165.04615327 185239.47102978
2112119.67255866185321.5357591612112078.38212878185447.700961565
#Sta/Elev= 30
       02404.316  37.9132400.796  80.525 2398.81 129.7212398.363 149.4672398.522
 179.0142399.419  212.212398.619 234.8242398.511 254.5222398.912  274.222398.429
 287.3512397.532 326.747 2397.47 346.4452396.963 398.7452396.592 402.5372396.441
 409.9312395.106 421.1782395.802 432.4252395.309 442.6372394.585 451.1692394.776
  456.61 2395.33 466.1652396.596 474.6872396.847 481.1612397.476  496.312400.122
 517.229    2405 544.4972411.951 554.8532414.147 596.2782422.188  629.062427.253
#Mann= 5 ,-1 , 0
       0    .035       0     190     .04       0  412.54      .1       0
 432.425    .045       0  456.61      .1       0
#XS Ineff= 2 , 0
          399.14 2399.98
Permanent Ineff=
       F       F
Bank Sta=432.425,456.61
XS Rating Curve= 0 ,0
Exp/Cntr(USF)=0,0
Exp/Cntr=0.5,0.3

Type RM Length L Ch R = 1 ,38750   ,35.4,35.8,37.1
XS GIS Cut Line= 4
2112180.36033666 184860.686522172112055.44300107185165.549690734
2112011.85865842185263.0409835012111976.30301047185402.969662531
#Sta/Elev= 30
       02395.522  32.7152392.419  61.7852390.307 114.9692387.903 129.1512387.603
  153.972387.503 182.3352387.867 213.7982389.148 285.1562391.013 302.8842390.838
 317.0662390.963 334.4562392.082 342.0542392.306 349.2422391.725 361.775 2391.94
   367.52391.722 374.3982391.149 384.1262391.667 392.3672392.038 403.1482393.254
  413.932393.868 431.8982395.396 438.9212396.614 449.0772398.985 459.2322400.722
 493.0832408.327 510.0082411.583 547.2442418.191 572.4352423.088 580.629 2424.35
#Mann= 5 ,-1 , 0
       0    .035       0     310     .04       0   367.5    .045       0
 384.126     .04       0  516.25      .1       0
#XS Ineff= 2 , 0
          362.93 2394.63  400.43         2394.54
Permanent Ineff=
       F       F
Bank Sta=367.5,384.126
XS Rating Curve= 0 ,0
Exp/Cntr(USF)=0,0
Exp/Cntr=0.5,0.3

Type RM Length L Ch R = 1 ,38714   ,59.7,60.1,60.5
XS GIS Cut Line= 4
2112179.02218624184860.0780101122112029.06300421185140.316650254
2111983.18474879185236.6609866352111941.89431891185390.353142291
#Sta/Elev= 30
       02395.554  29.0242392.706   54.372390.549  80.4172388.988 119.4232387.498
 164.3082387.028 184.6062387.291 225.5372388.911 288.7952389.734 311.121 2389.38
  322.182389.641 329.4482390.396 339.1592390.721 346.5442390.421 358.518 2390.94
 365.786  2390.6  369.422390.116  372.26  2390.6 376.6872391.348 387.5892391.962
 405.6222393.488 420.293  2394.1 427.3652394.995 430.7622395.601 447.748 2399.62
 468.1312403.449 491.9112408.504 556.4572419.692  576.842423.721 583.6912424.744
#Mann= 5 ,-1 , 0
       0    .035       0  327.84     .04       0 365.786    .045       0
  372.26     .04       0  434.55      .1       0
#XS Ineff= 2 , 0
          358.27 2394.85  380.39         2394.93
Permanent Ineff=
       F       F
Bank Sta=365.786,372.26
XS Rating Curve= 0 ,0
Exp/Cntr(USF)=0,0
Exp/Cntr=0.5,0.3

Type RM Length L Ch R = 1 ,38654   ,53.5,82.9,105.4
XS GIS Cut Line= 4
2112147.15424145184863.3472752042111982.41242735185103.574479364
2111929.38247794185206.5866799542111903.17227305185369.333766093
#Sta/Elev= 30
       0 2393.94    33.2 2390.34    70.1 2387.98   108.7 2386.88   165.4 2386.21
   205.5 2386.87   262.1 2387.24   296.4 2388.36   307.5 2389.27   318.6 2389.59
     326 2389.33   336.7 2389.76   341.6 2389.64   345.6 2389.21   348.9 2388.84
 352.9112389.149   361.1 2389.46   377.6 2390.78   390.3 2391.48   407.4 2393.32
   410.5 2393.87     416 2395.35   458.9  2407.3   476.9 2411.16   490.4 2413.06
   503.5 2415.34   520.1 2416.62   533.3 2418.43   546.7 2420.84     572 2424.69
#Mann= 5 ,-1 , 0
       0    .035       0     280     .04       0   345.6    .045       0
 352.911     .04       0  447.15      .1       0
#XS Ineff= 2 , 0
          330.09 2394.02
Permanent Ineff=
       F       F
Bank Sta=345.6,352.911
XS Rating Curve= 0 ,0
Exp/Cntr(USF)=0,0
Exp/Cntr=0.5,0.3

Type RM Length L Ch R = 1 ,38571   ,47.2,39,36
XS GIS Cut Line= 4
2112142.52058933184860.8785542642111913.53444708185118.203430927
2111852.58048223185103.5744793642111724.57715605185098.698162176
#Sta/Elev= 30
       0 2394.05    23.6 2391.21    38.1  2389.8    70.7 2387.76   114.8 2386.47
   159.7  2385.9   222.3 2385.68   247.6 2385.77   291.4 2386.65   304.6 2387.59
   312.4 2387.86   319.3 2388.69   326.6 2388.48   344.2 2388.97 363.1072388.111
   375.7 2387.17   379.1 2388.15   382.4    2389   399.3 2389.08   402.7 2389.58
   409.4 2391.91   412.6  2392.7   422.5 2394.39   442.2 2398.52   461.9 2402.85
   472.2 2405.43   481.6 2407.19   511.1 2411.01   528.2 2412.56   535.2 2412.86
#Mann= 5 ,-1 , 0
       0    .035       0     250     .04       0 363.107    .045       0
   379.1     .04       0  467.14      .1       0
#XS Ineff= 2 , 0
          351.58 2392.22  384.24         2392.22
Permanent Ineff=
       F       F
Bank Sta=363.107,379.1
XS Rating Curve= 0 ,0
Exp/Cntr(USF)=0,0
Exp/Cntr=0.5,0.3

Type RM Length L Ch R = 1 ,38532   ,84,79.6,75.9
XS GIS Cut Line= 4
2112140.68356419184856.2936235122111918.41076426185075.535655534
2111856.23772012185070.6593383472111720.31037851185091.383686394
#Sta/Elev= 30
       0  2394.5    35.4 2390.24    58.6 2388.47    80.6 2387.35   103.6  2386.9
   122.1 2386.12   241.8 2385.34   292.6 2386.13   306.8    2387   324.5 2387.18
   334.4 2387.58   337.7 2387.21  339.28 2386.72     341 2386.22   344.3  2385.8
   347.5 2386.74   350.8 2387.89   354.1  2388.2   360.7 2387.85   400.4  2387.8
     404 2388.67   409.7  2391.6   413.7 2393.17   430.3  2396.5   435.7  2397.9
   446.9 2401.39   456.8 2403.17   470.2 2406.05   496.1 2410.73   512.1 2412.18
#Mann= 5 ,-1 , 0
       0    .035       0     270     .04       0  339.28    .045       0
   347.5     .04       0  444.57      .1       0
#XS Ineff= 2 , 0
          333.52 2391.09  354.15         2391.09
Permanent Ineff=
       F       F
Bank Sta=339.28,347.5
XS Rating Curve= 0 ,0
Exp/Cntr(USF)=0,0
Exp/Cntr=0.5,0.3

Type RM Length L Ch R = 1 ,38453   ,158,148.7,139.8
XS GIS Cut Line= 4
2112137.65739765184852.5251854612111951.93544493184978.618851429
2111772.12124863185016.4103096342111702.02418906 185065.17348151
#Sta/Elev= 30
       0 2394.82    29.5 2391.18    41.9 2389.91    65.7 2388.06    89.5 2386.89
   133.1 2385.67   247.9 2385.22   257.9 2384.79     278 2384.43   304.8 2384.45
   308.8 2384.21   311.5 2383.92 318.3052384.205   325.4 2384.45   343.8 2384.16
   371.9 2385.26   383.6 2385.49   388.6 2385.96   395.3 2387.17   400.2 2387.68
   408.2 2387.98   420.3 2387.94   422.6 2388.67     425 2389.86   428.8  2392.3
   432.8 2393.96   448.6 2397.62   476.8 2406.33   482.7  2407.1   493.6 2408.97
#Mann= 5 ,-1 , 0
       0    .035       0   308.8    .045       0 318.305    .035       0
  394.48     .04       0  458.22      .1       0
#XS Ineff= 2 , 0
          220.92 2387.95
Permanent Ineff=
       F       F
Bank Sta=308.8,318.305
XS Rating Curve= 0 ,0
Exp/Cntr(USF)=0,0
Exp/Cntr=0.3,0.1

Type RM Length L Ch R = 1 ,38304   ,153.3,146.5,140.2
XS GIS Cut Line= 4
2112017.15618732184695.7924545432111889.76240079184813.433606696
2111729.45347324184991.4191840472111684.34753926 185061.51624362
#Sta/Elev= 30
       0 2404.02     8.2 2403.25    22.7 2401.06    26.8 2400.04    32.3 2398.11
    37.2    2397    66.2 2392.57    89.4 2386.86    97.5 2385.19   119.8 2382.12
   138.2 2381.41   166.1 2381.53   190.3 2381.04   212.7 2381.23   217.2 2380.93
   221.2 2380.54   225.6 2380.91   234.5 2381.27   281.3 2381.36   333.3 2382.66
   384.4 2385.26   393.4 2386.26     403    2388   421.8 2387.86   424.2 2388.51
   430.8 2391.67   445.5 2395.24   473.7 2404.33   486.6 2407.18   496.3 2408.65
#Mann= 6 ,-1 , 0
       0      .1       0     170    .035       0   217.2    .045       0
   225.6    .035       0   353.4     .04       0  482.94      .1       0
#XS Ineff= 2 ,-1
       0     149 2383.31  282.23 496.295 2383.91
Permanent Ineff=
       F       F
Bank Sta=217.2,225.6
XS Rating Curve= 0 ,0
Exp/Cntr(USF)=0,0
Exp/Cntr=0.3,0.1

Type RM Length L Ch R = 1 ,38158   ,352,345.6,335.7
XS GIS Cut Line= 4
2111901.79848122184266.1540194042111787.41383941184585.567736171
2111679.50379996184948.145468718 2111656.6034647185060.953347025
#Sta/Elev= 30
       0 2482.27    23.1 2478.83      65  2471.4   155.6 2451.24   188.1  2443.1
   204.4 2438.52   242.7 2426.14   285.6 2410.89   319.4 2399.88   340.2 2392.53
   355.4 2388.31   367.6 2383.79   394.9  2378.7   432.7 2377.34 535.3582378.311
   542.2 2378.01  549.052378.386   555.8 2379.07   571.7 2379.06   631.2 2381.58
   682.5 2385.27     712 2386.73   722.3 2388.32   743.6 2388.14   750.3 2389.75
   766.8 2390.45   790.4 2393.36   803.8 2395.85   820.6    2400   832.7  2403.6
#Mann= 9 ,-1 , 0
       0     .12       0      30      .1       0     100     .12       0
     200      .1       0  409.28    .035       0 535.358    .045       0
  549.05    .035       0  659.28     .04       0  817.57      .1       0
#XS Ineff= 2 ,-1
       0  438.83 2381.16   556.5 832.681 2379.98
Permanent Ineff=
       F       F
Bank Sta=535.358,549.05
XS Rating Curve= 0 ,0
Exp/Cntr(USF)=0,0
Exp/Cntr=0.3,0.1

Type RM Length L Ch R = 1 ,37812   ,347.3,350.5,356.6
XS GIS Cut Line= 3
     2111312.755      184151.107     2111401.813      184690.524
     2111508.004      185226.332
#Sta/Elev= 30
       0 2481.48    55.6 2465.74   125.4  2441.8   205.2 2416.29   271.7 2392.76
   302.1 2384.14   311.6 2380.59   324.9  2377.4   354.8 2372.32   378.1 2371.36
   544.4  2371.7     551 2370.69  558.772371.744   601.2 2372.08   634.7 2373.35
   661.4 2377.94   718.3 2393.69   745.2 2394.39   751.7 2395.32   761.4 2398.01
   771.8 2397.28   795.2 2397.88   835.3 2401.47   845.4 2403.28     865 2404.02
   885.5 2406.45   915.6 2407.53   979.2 2411.63  1032.7 2417.44  1092.9 2419.68
#Mann= 6 ,-1 , 0
       0      .1       0     410    .035       0   544.4    .045       0
  558.77    .035       0  606.72     .04       0  806.72      .1       0
#XS Ineff= 2 , 0
          398.58 2373.54  582.08         2373.42
Permanent Ineff=
       F       F
Bank Sta=544.4,558.77
XS Rating Curve= 0 ,0
Exp/Cntr=0.3,0.1

Type RM Length L Ch R = 1 ,37461   ,136.9,136.6,139.1
XS GIS Cut Line= 3
       2111067.4      184160.193     2111053.461      184705.996
     2111034.263      185251.702
#Sta/Elev= 30
       0 2453.44    12.9 2451.34    22.8 2447.84    48.9 2440.57   104.8  2426.8
   111.4 2426.04   160.9 2411.64   193.4 2403.47   242.7 2392.18   255.8  2388.4
   334.5 2372.83   344.4 2368.96   347.7 2368.36   372.4 2366.93     545 2365.51
   551.2    2365   579.8 2365.56   598.9 2365.85   627.4 2367.73   640.1 2367.26
   652.9 2369.62     689 2373.79   700.4 2376.48   715.3 2383.02   734.7 2390.08
   764.5 2399.39   833.5 2413.27   948.4 2431.64  1027.4 2445.97    1092 2459.62
#Mann= 6 ,-1 , 0
       0      .1       0     400    .035       0     545    .045       0
   579.8    .035       0  595.98     .04       0  695.98      .1       0
#XS Ineff= 2 , 0
          408.93 2368.72  627.72         2368.56
Permanent Ineff=
       F       F
Bank Sta=545,579.8
XS Rating Curve= 0 ,0
Exp/Cntr=0.5,0.3

Type RM Length L Ch R = 1 ,37325   ,28.6,28.5,28.5
XS GIS Cut Line= 2
     2110924.719      184165.855     2110909.094      185249.188
#Sta/Elev= 30
       0 2434.32    46.6 2418.27    72.9 2411.77    89.3 2408.48   105.7 2406.38
   115.5 2406.51   128.7 2405.47   164.8 2400.82   253.3 2382.71   276.3 2378.91
   288.1 2376.08   312.4 2373.53   332.1 2369.18     356 2367.15   384.6 2365.73
   531.5 2363.93   538.8 2363.08   543.8 2363.81   591.3 2365.18     611 2366.45
   630.7 2366.39   637.2 2365.49   676.3 2369.62   702.9 2375.76   725.8 2383.52
   791.5 2403.48   857.1 2419.45   899.7 2427.59  1037.5  2450.7  1083.4 2461.32
#Mann= 6 ,-1 , 0
       0      .1       0     390    .035       0   531.5    .045       0
   543.8    .035       0     590     .04       0     690      .1       0
#XS Ineff= 2 , 0
          512.45 2367.93  559.27         2367.93
Permanent Ineff=
       F       F
Bank Sta=531.5,543.8
XS Rating Curve= 0 ,0
Exp/Cntr=0.5,0.3

Type RM Length L Ch R = 1 ,37296   ,143.2,141,138.5
XS GIS Cut Line= 2
     2110896.247      184163.772     2110880.622      185247.105
#Sta/Elev= 30
       0 2433.18    91.4 2404.26   107.8 2403.29   124.2 2405.85   130.7 2405.62
     220 2387.79   258.9 2382.08   330.9 2368.63   360.4 2366.14   393.2 2364.93
   514.6 2364.02  535.25  2363.2   537.6 2362.87   544.2 2363.19   567.1 2363.85
   583.5 2365.23   596.7 2364.45   609.8 2366.22   642.6 2365.79   678.7 2369.41
   695.1 2372.08     728 2381.71   760.7 2392.37   816.5 2408.35   836.2 2413.09
   865.7 2419.61   914.9 2429.09  1039.6 2449.56  1065.9 2456.34  1083.4 2461.87
#Mann= 6 ,-1 , 0
       0      .1       0     390    .035       0     490     .04       0
  535.25    .045       0   544.2     .04       0     690      .1       0
#XS Ineff= 2 , 0
          523.55  2367.6  559.84         2367.51
Permanent Ineff=
       F       F
Bank Sta=535.25,544.2
XS Rating Curve= 0 ,0
Exp/Cntr=0.5,0.3

Type RM Length L Ch R = 1 ,37155   ,152.9,150.5,147.7
XS GIS Cut Line= 4
2110675.84392419184159.4318610162110728.28820337184530.038100521
2110775.48805462184932.1109075312110824.43604852185252.021010501
#Sta/Elev= 30
       0 2431.59    27.1 2426.11      90 2418.22     153 2406.68   196.1 2396.83
   242.4 2384.92   270.4 2376.36   290.8 2371.07   302.1  2367.1   331.9 2363.03
   386.8 2361.71   536.42362.487   543.5 2361.86   550.1 2362.44   614.4 2366.16
   626.2 2368.39   649.2  2367.3   659.1 2370.04   678.9 2371.66   725.1 2377.22
   781.3 2391.63   808.7 2397.17   831.8 2400.34   854.8 2404.48   900.7 2415.71
   923.9 2420.34   955.5 2429.35   990.4 2436.48  1053.6  2447.6  1102.8 2460.09
#Mann= 6 ,-1 , 0
       0      .1       0   404.3    .035       0   536.4    .045       0
   550.1    .035       0   594.3     .04       0   694.3      .1       0
#XS Ineff= 2 , 0
           365.9 2371.22   591.4         2371.66
Permanent Ineff=
       F       F
Bank Sta=536.4,550.1
XS Rating Curve= 0 ,0
Exp/Cntr(USF)=0,0
Exp/Cntr=0.5,0.3

Type RM Length L Ch R = 1 ,37005   ,30.7,30.7,30.8
XS GIS Cut Line= 2
     2110445.306      184151.128     2110756.563      185259.141
#Sta/Elev= 30
       0 2449.92    50.1 2449.62   131.9 2442.94   292.1 2403.13   332.5 2390.94
   388.3 2372.14   430.9 2363.57   462.4 2360.54   554.5  2362.1  559.962361.195
   564.7 2360.33   573.82361.183   646.5 2366.97   666.9 2370.07   690.8 2369.11
   704.4 2372.91   743.2 2375.81   762.3 2378.98   789.6  2379.5   806.6 2381.35
   848.6 2391.74     885 2399.21   905.5 2401.61   931.1 2402.36  1031.5 2418.49
  1065.6 2428.88  1089.5 2432.78  1109.9 2433.92    1127 2436.49  1150.9 2444.83
#Mann= 6 ,-1 , 0
       0      .1       0     420    .035       0  559.96    .045       0
   573.8    .035       0     630     .04       0     830      .1       0
#XS Ineff= 2 , 0
          553.66 2367.19  580.94         2367.28
Permanent Ineff=
       F       F
Bank Sta=559.96,573.8
XS Rating Curve= 0 ,0
Exp/Cntr=0.5,0.3

Type RM Length L Ch R = 1 ,36974   ,218.6,212,205.3
XS GIS Cut Line= 2
     2110417.528      184165.885     2110728.785      185273.898
#Sta/Elev= 30
       0  2452.3      62 2452.24    92.7 2450.23   123.4 2446.47   290.4 2404.96
   402.8 2372.33   446.8 2361.84   490.4 2360.26   554.12361.003   559.6  2359.7
  568.992361.014   614.4 2363.33   668.6 2369.38   692.5 2368.61   704.8 2372.71
   716.3 2372.87     730  2375.8   743.6 2375.17   784.2 2381.08   822.1 2393.17
   874.2 2407.39   912.1 2414.81   978.9 2422.61  1012.8 2429.94    1023 2430.37
  1046.9 2426.18  1076.4  2427.2  1122.5 2436.15  1143.8 2436.21  1150.9  2438.1
#Mann= 7 ,-1 , 0
       0      .1       0     410    .035       0   554.1    .045       0
  568.99    .035       0     610      .1       0     710     .04       0
     810      .1       0
#XS Ineff= 2 , 0
           550.3 2365.08  573.24          2364.9
Permanent Ineff=
       F       F
Bank Sta=554.1,568.99
XS Rating Curve= 0 ,0
Exp/Cntr=0.5,0.3

Type RM Length L Ch R = 1 ,36762   ,341.8,350,357.1
XS GIS Cut Line= 3
     2110069.723      184375.775      2110391.72      184815.892
     2110731.293      185287.932
#Sta/Elev= 30
       0  2470.4    49.7 2472.34    74.1 2470.46   181.9 2468.61   228.6 2466.45
   244.1 2464.09     345 2432.98   413.1  2409.4   424.8 2403.61   464.8 2388.79
   513.1 2366.01   537.5 2358.51   543.1 2357.27  550.732358.439   598.6 2358.26
   624.5 2359.18   658.8 2362.66   683.3 2362.09   691.1 2366.12   731.6    2379
   817.2 2402.98   919.5 2430.54   986.2 2445.08  1002.9 2446.82  1030.6 2446.52
    1057 2443.26  1087.6  2442.8  1110.5 2438.58  1118.1 2440.05  1126.8 2444.07
#Mann= 5 ,-1 , 0
       0      .1       0   537.5    .045       0  550.73      .1       0
  585.33     .04       0  705.33      .1       0
Bank Sta=537.5,550.73
XS Rating Curve= 0 ,0
Exp/Cntr=0.3,0.1

Type RM Length L Ch R = 1 ,36412   ,264,256.5,236.9
XS GIS Cut Line= 3
     2109986.584      184421.473     2110135.847      185025.651
     2110169.876      185558.654
#Sta/Elev= 30
       0 2456.15   109.2 2448.13   122.7 2445.83   136.5 2444.52   159.8 2440.74
   186.9  2437.3   227.4 2434.04   339.8 2420.31   416.7 2413.19   457.2 2411.29
   487.7 2407.93   494.7 2406.47   507.8 2401.65   534.6 2389.71   570.1 2375.49
  614.112352.139   616.1  2351.2   619.5 2350.84  627.272352.137   645.8 2353.85
   672.1 2353.78   678.7 2356.84   695.7  2360.3   721.4 2368.11   816.8 2404.53
   882.5 2433.39   987.7 2473.46  1040.3 2495.96  1102.8 2518.27  1156.4  2539.6
#Mann= 5 ,-1 , 0
       0      .1       0  614.11    .045       0  627.27      .1       0
  642.34     .04       0  742.34      .1       0
#XS Ineff= 2 , 0
                          659.87         2355.44
Permanent Ineff=
       F       F
Bank Sta=614.11,627.27
XS Rating Curve= 0 ,0
Exp/Cntr=0.5,0.3

Type RM Length L Ch R = 1 ,36156   ,47.8,56.9,58.7
XS GIS Cut Line= 4
     2109966.411      184419.189     2109876.568      184959.554
     2109922.141      184986.898     2109867.453      185522.054
#Sta/Elev= 30
       0 2453.02    86.5 2441.33   169.6 2425.17   206.2 2420.33   299.3 2403.02
   345.9 2397.44   422.4 2385.48   435.7 2382.16   464.2    2372   482.2 2364.14
   502.2 2353.63   522.1 2346.75   535.4 2343.52   573.1 2341.74   576.3 2341.23
     581 2341.85   623.9 2342.82   631.5 2346.46   660.1 2352.48   680.6 2360.25
     736 2384.68   752.5 2391.06   775.6 2397.84   805.3 2410.48   874.5 2445.69
   904.6 2465.73   930.8  2480.7   986.6 2507.93  1059.2 2536.42  1138.9 2558.05
#Mann= 5 ,-1 , 0
       0      .1       0     540     .04       0   573.1    .045       0
     581     .04       0  660.93      .1       0
#XS Ineff= 2 , 0
           565.8  2346.4  585.67         2346.56
Permanent Ineff=
       F       F
Bank Sta=573.1,581
XS Rating Curve= 0 ,0
Exp/Cntr=0.5,0.3

Type RM Length L Ch R = 1 ,36099   ,253.2,262.9,281.5
XS GIS Cut Line= 4
     2109935.161      184413.981     2109838.807      184982.991
      2109884.38      185010.335     2109833.599      185524.658
#Sta/Elev= 30
       0 2449.95    15.2 2446.93    48.5 2443.44   304.7 2397.72   427.9 2379.35
   444.5 2375.13   527.7 2341.71   544.3 2339.63   564.3 2340.34   567.6 2339.94
  574.952336.025   577.6 2334.92   587.3  2336.2   603.6 2337.38   622.7 2348.13
   630.3 2349.04   642.8 2353.05     722 2383.84   769.4 2404.47     811 2412.92
   840.6 2424.59   886.8 2446.36   913.2 2460.98   965.9 2493.91   996.2 2510.21
  1021.8 2522.39  1051.6 2533.28  1079.1 2541.39  1124.1 2552.97  1147.1 2557.25
#Mann= 5 ,-1 , 0
       0      .1       0     540     .04       0  574.95    .045       0
   587.3     .04       0  670.26      .1       0
#XS Ineff= 2 , 0
          571.86  2341.3  590.82         2341.43
Permanent Ineff=
       F       F
Bank Sta=574.95,587.3
XS Rating Curve= 0 ,0
Exp/Cntr=0.5,0.3

Type RM Length L Ch R = 1 ,35836   ,248.4,267.6,286.5
XS GIS Cut Line= 4
2109742.33575487184379.6978335522109667.16562139184708.348649717
2109567.52149095185120.9103125622109506.33649858185439.072272892
#Sta/Elev= 30
       0 2429.05      54 2422.92   215.5  2392.7   319.8 2368.86     360 2357.37
   424.4 2340.77   463.1 2332.26   471.5 2329.82   488.5 2322.72   498.7 2321.01
   508.8  2321.9   525.4 2321.47  530.272319.792   535.8  2318.5  542.282319.793
     556 2324.71   589.8 2328.53   614.4 2335.74   656.3 2353.17   701.2    2370
   777.8 2404.65     812 2421.29   829.6    2428   855.5 2433.88   925.6 2444.16
   955.7 2447.23  1014.6 2456.48    1026 2460.29  1049.3 2470.13  1085.6 2486.78
#Mann= 5 ,-1 , 0
       0      .1       0  487.14     .04       0  530.27    .045       0
  542.28     .04       0  587.14      .1       0
#XS Ineff= 2 , 0
          509.88 2326.92
Permanent Ineff=
       F       F
Bank Sta=530.27,542.28
XS Rating Curve= 0 ,0
Exp/Cntr(USF)=0,0
Exp/Cntr=0.5,0.3

Type RM Length L Ch R = 1 ,35568   ,52.9,44.5,31.8
XS GIS Cut Line= 4
     2109519.276      184320.513     2109387.983      184826.155
      2109348.92      184832.666     2109309.858      185399.072
#Sta/Elev= 30
       0 2413.65   135.8 2395.65   210.4 2383.31   244.3 2376.72   318.9    2361
   393.4 2340.98     468 2312.84  527.072307.743   540.4 2306.77  548.062307.743
     555 2309.69     562 2309.69   581.6 2315.87   611.2  2319.6     631 2323.63
   663.8 2334.93   714.4 2349.77   735.9 2357.43   762.5  2369.7   788.8 2383.22
     822 2397.42     862 2413.54   890.8  2422.9   917.4 2433.32   956.5 2442.94
     996 2457.31  1051.9    2470  1080.5 2480.97  1107.4 2489.83  1129.8 2493.96
#Mann= 5 ,-1 , 0
       0      .1       0     450     .04       0  527.07    .045       0
  548.06     .04       0  682.01      .1       0
#XS Ineff= 2 , 0
           518.1 2311.13  555.34         2311.03
Permanent Ineff=
       F       F
Bank Sta=527.07,548.06
XS Rating Curve= 0 ,0
Exp/Cntr=0.5,0.3

Type RM Length L Ch R = 1 ,35524   ,155.6,150.2,136.1
XS GIS Cut Line= 4
     2109489.979      184311.832     2109363.026      184796.859
     2109323.963      184803.369     2109282.731      185399.072
#Sta/Elev= 30
       0 2412.07    83.8 2402.03   199.1 2385.01   312.5 2364.21     382 2347.89
     406 2343.54   430.8 2334.73     467 2318.37   478.5 2314.11   490.8 2310.76
   520.6 2307.57  527.332305.346     532 2304.18  541.152305.346   547.2 2308.22
   573.5 2308.32   583.4 2312.76   622.8 2316.72   636.2 2319.71   705.1 2341.58
   790.6 2378.56   856.3 2404.33   899.1 2418.29   925.4 2428.43   968.2 2441.14
   995.7 2451.63  1066.8 2470.03  1094.1 2480.13  1116.1 2484.16  1138.1 2486.16
#Mann= 5 ,-1 , 0
       0      .1       0     460     .04       0  527.33    .045       0
  541.15     .04       0  690.97      .1       0
#XS Ineff= 2 , 0
          523.34 2310.28  545.01         2310.28
Permanent Ineff=
       F       F
Bank Sta=527.33,541.15
XS Rating Curve= 0 ,0
Exp/Cntr=0.5,0.3

Type RM Length L Ch R = 1 ,35374   ,270,263.3,255.8
XS GIS Cut Line= 3
     2109169.602      184275.693     2109187.347      184813.078
     2109265.606      185405.225
#Sta/Elev= 30
       0 2407.91    74.6 2404.05   205.9 2382.13   225.1 2378.43   235.5 2373.91
     265 2372.63   298.2  2365.5   327.4 2356.99   370.1 2348.92   425.3 2333.77
   468.5 2324.76   494.8 2315.85   501.4 2312.63   518.1 2302.17  524.432300.783
   537.5 2299.55  551.612300.783   573.9 2305.19   603.7 2304.89   610.3 2307.87
   646.7 2317.41   686.4 2330.71   759.2 2363.43   782.4 2371.91   888.3 2414.54
     928 2426.09   974.3 2441.73  1060.3 2466.21  1115.4 2476.32    1135 2481.03
#Mann= 5 ,-1 , 0
       0      .1       0  524.43    .045       0  551.61      .1       0
  577.68     .04       0  677.68      .1       0
Bank Sta=524.43,551.61
XS Rating Curve= 0 ,0
Exp/Cntr=0.3,0.1

Type RM Length L Ch R = 1 ,35110   ,172.6,156.4,134.8
XS GIS Cut Line= 2
     2108735.443      184448.145     2109241.086      185409.516
#Sta/Elev= 30
       0 2417.59    89.6 2389.15   169.1 2372.46   237.9 2355.88     259 2348.38
   271.2 2339.32   293.5 2338.83   315.7 2327.85   330.5  2326.5   348.8 2320.61
   367.6 2317.61   392.6 2311.41   415.8 2310.96   441.8 2305.86   449.2 2302.46
  458.942293.733     464 2292.46   471.4 2293.53   494.6 2297.18   506.7 2295.81
   564.1 2295.45   572.3 2298.11   620.9 2305.32   650.1 2312.17   756.8 2355.86
   815.3    2378     884 2410.14   912.2 2421.63   997.8 2444.92  1086.2 2473.96
#Mann= 4 ,-1 , 0
       0      .1       0  458.94    .045       0   471.4     .04       0
     570      .1       0
#XS Ineff= 2 , 0
                          495.13         2307.95
Permanent Ineff=
       F       F
Bank Sta=458.94,471.4
XS Rating Curve= 0 ,0
Exp/Cntr=0.5,0.3

Type RM Length L Ch R = 1 ,34954   ,43.7,43.1,45.7
XS GIS Cut Line= 4
     2108704.895      184455.185     2108822.083      184964.734
     2108863.749       184966.47     2108992.221      185444.768
#Sta/Elev= 30
       0 2416.24    57.3 2395.05    97.7 2382.08   124.6 2376.24   178.5 2366.69
   208.8 2359.36   262.7 2341.35   269.4 2337.64   276.1 2331.93   279.5 2330.14
   299.7 2329.19   316.5    2321   336.7 2314.85   372.8 2307.45   407.4 2302.23
   441.1 2299.74   464.7 2296.51   488.2 2291.56  532.752288.762   539.3 2287.32
  552.482288.762     563 2290.23   595.4 2290.29   605.9 2292.54   622.9 2293.81
   721.4 2310.66   758.4 2323.51   793.5 2338.46   900.6 2379.24  1059.8 2426.79
#Mann= 5 ,-1 , 0
       0      .1       0     510     .04       0  532.75    .045       0
  552.48     .04       0  654.55      .1       0
#XS Ineff= 2 , 0
          529.62 2295.99  557.89         2295.93
Permanent Ineff=
       F       F
Bank Sta=532.75,552.48
XS Rating Curve= 0 ,0
Exp/Cntr=0.5,0.3

Type RM Length L Ch R = 1 ,34911   ,239.9,273,298.1
XS GIS Cut Line= 4
     2108684.756      184467.251     2108807.152      185005.445
     2108848.819      185007.182     2108972.951      185461.175
#Sta/Elev= 30
       0 2412.41    47.2 2394.47    81.9 2382.93   102.2  2377.9   125.7 2374.45
     166 2366.52   190.6 2360.56   256.9    2340     267  2335.2   277.1 2327.73
   300.6 2327.33     304 2325.87   314.1 2318.63   337.6 2311.97   408.3 2300.27
   435.2 2298.28   499.1 2288.89   557.1 2288.47   563.92287.655   570.2 2286.25
   575.32287.655   580.1 2288.83   608.7 2290.57   643.9 2294.41   701.7 2305.51
   752.7 2326.71   827.7  2356.2   870.5 2371.22  1004.4 2412.25  1064.3 2427.81
#Mann= 5 ,-1 , 0
       0      .1       0     500     .04       0   563.9    .045       0
   575.3     .04       0  633.64      .1       0
#XS Ineff= 2 , 0
          561.77 2292.25  577.91            2292
Permanent Ineff=
       F       F
Bank Sta=563.9,575.3
XS Rating Curve= 0 ,0
Exp/Cntr=0.5,0.3

Type RM Length L Ch R = 1 ,34638   ,183.9,190.4,196.1
XS GIS Cut Line= 4
2108647.99846275184467.1049655112108604.29489677184958.333047119
2108586.81347037185222.3025856352108581.56904246185577.175541387
#Sta/Elev= 30
       0 2412.64      54 2393.27   123.2 2377.27   248.3 2340.29     291 2329.61
   304.3 2324.82   317.5 2314.13     334 2314.47   360.3  2303.8   406.4 2300.56
   478.9 2287.88   505.2 2287.68   554.5 2282.42   641.3 2280.19   646.6 2279.88
   651.9 2280.47   688.2 2283.07   709.1 2280.88   807.6 2284.04   817.5 2286.51
   837.1 2297.53   873.2 2305.76   925.7  2302.2   958.5 2309.03   968.4 2313.36
   994.6  2330.7  1010.6 2333.09    1047 2333.63  1060.3 2328.24  1112.6 2321.83
#Mann= 9 ,-1 , 0
       0      .1       0     390     .06       0     490     .04       0
  583.17      .1       0   641.3    .045       0   651.9      .1       0
  683.17     .08       0  977.72     .06       0 1077.72      .1       0
#XS Ineff= 2 , 0
                           753.8         2298.19
Permanent Ineff=
       F       F
Bank Sta=641.3,651.9
XS Rating Curve= 0 ,0
Exp/Cntr(USF)=0,0
Exp/Cntr=0.5,0.3

Type RM Length L Ch R = 1 ,34448   ,42.8,40.1,47.8
XS GIS Cut Line= 2
     2108608.541      184459.439     2108233.541      185639.994
#Sta/Elev= 30
       0 2415.36    54.1 2398.19   202.8 2362.54   305.4 2327.75   346.7 2311.74
   360.5 2303.07   381.2 2301.97   412.1 2294.31   486.5 2284.74   501.6 2280.46
   529.3 2280.66   650.3 2275.98   656.6 2274.92  683.342275.979   701.8 2276.36
   725.6 2279.56   752.9 2280.78   773.6 2285.24   797.7  2288.2   819.3 2282.54
   894.1 2284.41   910.8 2283.25     920 2286.64   942.1 2298.56   990.5 2317.45
  1021.4 2328.88  1073.7 2345.94  1124.7 2356.11  1203.4  2363.8  1238.7 2372.66
#Mann= 5 ,-1 , 0
       0      .1       0     410     .06       0     510      .1       0
   650.3    .045       0  683.34      .1       0
#XS Ineff= 2 , 0
          635.18 2280.98  689.05         2280.83
Permanent Ineff=
       F       F
Bank Sta=650.3,683.34
XS Rating Curve= 0 ,0
Exp/Cntr=0.5,0.3

Type RM Length L Ch R = 1 ,34407   ,210.6,208.3,204.3
XS GIS Cut Line= 2
     2108571.735      184448.327     2108196.735      185628.883
#Sta/Elev= 30
       0 2419.71    89.9 2393.17   203.5  2365.7     262 2345.36   320.1 2327.54
   362.6 2310.02   382.5 2298.16   396.3  2298.7     431 2290.31   492.7 2282.66
   509.9 2278.57   599.4 2278.44   621.2 2276.72  635.072273.751   647.3 2272.41
  652.672273.752   688.9 2277.15     744 2278.76   761.2 2280.97   788.4 2279.37
   836.9 2280.65   852.6 2279.13   929.5 2304.23    1009 2334.46  1050.3 2346.23
  1080.1 2351.37  1143.3 2353.88  1187.8  2357.8  1208.7 2361.58  1238.7 2370.95
#Mann= 5 ,-1 , 0
       0      .1       0     420     .06       0     530      .1       0
  635.07    .045       0  652.67      .1       0
#XS Ineff= 2 , 0
          630.79 2277.92  655.43         2277.97
Permanent Ineff=
       F       F
Bank Sta=635.07,652.67
XS Rating Curve= 0 ,0
Exp/Cntr=0.5,0.3

Type RM Length L Ch R = 1 ,34199   ,232.9,229.6,223.5
XS GIS Cut Line= 4
2108170.75552225184451.371681758  2108186.488806184933.859050171
2108184.74066336185180.3471622942108163.76295169185622.627250006
#Sta/Elev= 30
       0 2410.54    13.7  2401.3    69.5 2379.19   102.4 2372.38   135.2 2363.55
   250.3 2319.44   332.1 2296.33   364.7 2288.75   397.8 2283.93   443.8 2279.08
   476.6 2277.22   486.4 2273.86   525.8 2272.98  547.242268.611   558.6 2267.58
  566.152268.611   594.7 2270.51   640.6 2269.96     699 2272.16   712.8 2276.38
   752.2 2295.59   781.9 2307.38   850.6 2327.41   903.3 2340.11   922.7 2343.61
   955.8 2345.62  1024.8 2342.31  1097.1 2349.28  1126.6 2355.12    1172 2370.57
#Mann= 5 ,-1 , 0
       0      .1       0  502.74     .04       0  547.24    .045       0
  566.15     .04       0  592.74      .1       0
#XS Ineff= 2 , 0
                          594.84         2280.49
Permanent Ineff=
       F       F
Bank Sta=547.24,566.15
XS Rating Curve= 0 ,0
Exp/Cntr(USF)=0,0
Exp/Cntr=0.3,0.1

Type RM Length L Ch R = 1 ,33969   ,158,156.4,155
XS GIS Cut Line= 3
     2107881.446      184530.972     2107978.237      185097.025
     2108104.413       185623.07
#Sta/Elev= 30
       0 2381.77    36.4  2377.9    59.7 2372.42      73 2367.61   101.2 2354.62
   186.1 2308.19   219.4 2294.78   325.9 2277.73   385.8 2271.51   432.4 2269.01
   442.4 2265.23     479 2266.94   553.3 2265.27  567.372260.922   573.2 2259.62
  581.352260.923   612.7 2263.51   626.2 2266.53   668.2 2287.76   694.8 2299.44
     724 2309.62   754.4 2317.61   781.4 2321.81   801.4 2322.17     878  2315.2
   896.1 2310.64   932.4 2323.87   993.9 2335.73  1024.3 2343.44  1115.2 2372.22
#Mann= 5 ,-1 , 0
       0      .1       0     430     .04       0     530      .1       0
  567.37    .045       0  581.35      .1       0
#XS Ineff= 2 , 0
          541.55 2275.67
Permanent Ineff=
       F       F
Bank Sta=567.37,581.35
XS Rating Curve= 0 ,0
Exp/Cntr=0.5,0.3

Type RM Length L Ch R = 1 ,33813   ,32.4,31.7,33.9
XS GIS Cut Line= 4
2107821.21440155 184535.614675542107788.64650418184983.069265463
2107856.61428999185225.2045024162107937.32603564185628.763230669
#Sta/Elev= 30
       0 2373.22    37.9  2366.5    54.3 2361.59    80.6 2350.16   110.2 2335.37
   146.4 2322.15   185.9 2304.92   218.5 2295.12   258.3 2286.74   284.6  2278.9
   307.2 2275.31   347.8 2271.29   396.4 2262.98     426 2262.31   435.9 2259.77
     507 2260.04   534.4 2257.81   571.7 2258.35   578.6 2256.89   587.4 2258.32
   622.8 2258.13   646.7  2259.5   670.6 2263.39   707.9  2264.4     742  2272.2
   798.2 2280.24   863.3 2301.39   915.3 2315.48  1029.1  2340.2  1111.7 2356.32
#Mann= 7 ,-1 , 0
       0      .1       0     420     .04       0  518.64      .1       0
   571.7    .045       0   587.4      .1       0  710.13     .06       0
  720.13      .1       0
#XS Ineff= 2 , 0
          567.86 2264.73  591.88         2264.68
Permanent Ineff=
       F       F
Bank Sta=571.7,587.4
XS Rating Curve= 0 ,0
Exp/Cntr(USF)=0,0
Exp/Cntr=0.5,0.3

Type RM Length L Ch R = 1 ,33781   ,152.2,161.9,168.5
XS GIS Cut Line= 4
2107805.63845063184534.1986800022107761.74258896184985.901256539
2107828.29437924185256.356404246 2107901.9261472185630.179226207
#Sta/Elev= 30
       0 2371.34    36.1 2364.64    55.8 2359.11   105.3 2336.86   135.5 2326.92
   171.2 2311.62   200.9 2300.71   293.2 2276.76   339.3  2271.5   359.1 2268.68
   378.9 2264.63   411.8 2261.97   434.9 2258.69     448 2259.25   491.9  2257.5
     569 2257.21   576.3 2256.59     584 2257.24   637.2 2258.44   670.9 2262.88
   717.7 2264.47   748.4 2269.55   755.2 2269.62   761.9 2271.51     792 2276.77
   848.5 2293.89   882.2 2302.74   915.7 2310.17   999.3 2326.33  1113.4  2345.6
#Mann= 5 ,-1 , 0
       0      .1       0     420     .04       0  513.83      .1       0
     569    .045       0     584      .1       0
#XS Ineff= 2 , 0
          564.95 2261.91  589.38         2262.02
Permanent Ineff=
       F       F
Bank Sta=569,584
XS Rating Curve= 0 ,0
Exp/Cntr(USF)=0,0
Exp/Cntr=0.5,0.3

Type RM Length L Ch R = 1 ,33619   ,152.5,155.8,158.7
XS GIS Cut Line= 3
     2107781.135      184529.894     2107634.555      185102.417
     2107519.888      185628.619
#Sta/Elev= 30
       0 2369.09    31.3 2362.78    51.7    2357      89 2340.65   146.5 2323.59
   170.2 2314.46   181.2 2311.23   231.1 2291.74   245.2 2287.78   281.9  2279.6
   363.9 2266.91   436.7  2259.4   451.3 2256.83   471.6  2257.7   487.9  2255.5
     563 2256.33   576.9 2253.59  584.322251.085   590.4 2249.68   593.5 2249.97
  596.082251.084   612.4 2259.11   627.1 2264.01   684.2 2279.87     805 2318.67
   875.6 2337.66   912.5 2346.22   972.9 2358.18  1056.9 2371.72  1129.5 2381.05
#Mann= 5 ,-1 , 0
       0      .1       0     430     .04       0     540      .1       0
  584.32    .045       0  596.08      .1       0
#XS Ineff= 2 , 0
          560.46 2266.14
Permanent Ineff=
       F       F
Bank Sta=584.32,596.08
XS Rating Curve= 0 ,0
Exp/Cntr=0.3,0.1

Type RM Length L Ch R = 1 ,33464   ,190.7,194.2,202
XS GIS Cut Line= 4
2107736.25466928184511.5427513982107550.75925384184917.933470728
2107454.47155727185127.5008103122107263.31215968185492.827659047
#Sta/Elev= 30
       0 2368.39    21.1 2364.76      68 2351.76   122.1 2331.05   172.6 2317.97
   197.7 2310.23   219.4 2301.39   241.1 2294.21   291.6 2281.29   314.1 2272.85
   338.4 2266.57   370.9 2261.58   452.8 2254.46   518.9 2254.23   540.5 2250.61
   569.4 2249.92  578.522248.467   583.8 2246.69  595.352248.468   682.8 2250.52
   711.1 2253.14   729.6 2257.25   741.1 2261.14   770.3 2274.96   845.6 2316.37
   884.5 2332.28   908.8 2338.49   961.3 2343.89    1011 2344.66  1089.7 2342.63
#Mann= 4 ,-1 , 0
       0      .1       0     420     .04       0  578.52    .045       0
  595.35      .1       0
Bank Sta=578.52,595.35
XS Rating Curve= 0 ,0
Exp/Cntr(USF)=0,0
Exp/Cntr=0.3,0.1

Type RM Length L Ch R = 1 ,33269   ,332.2,325,310.1
XS GIS Cut Line= 3
     2107693.303      184482.482     2107340.016       184929.44
     2106932.019      185287.829
#Sta/Elev= 30
       0 2368.46    52.5 2358.35   128.4 2335.41   190.1 2320.28   237.1 2304.43
   311.8 2284.63   375.1 2262.78   426.6 2254.45   447.6 2254.22   522.3 2246.37
  557.832244.828   565.7 2243.17   575.1 2244.91   657.4 2243.75   676.5 2244.75
   701.3 2251.64   721.2 2253.41   749.8 2259.39   767.3 2261.37     811 2260.13
   824.1 2255.84   832.8  2259.8     855 2259.42   876.5  2260.9     925 2287.46
     942 2293.09   954.8 2300.18  1017.7 2327.87  1064.2  2345.2  1112.8 2359.34
#Mann= 5 ,-1 , 0
       0      .1       0     370     .04       0     530      .1       0
  557.83    .045       0   575.1      .1       0
#XS Ineff= 2 , 0
                          632.93         2247.28
Permanent Ineff=
       F       F
Bank Sta=557.83,575.1
XS Rating Curve= 0 ,0
Exp/Cntr=0.3,0.1

Type RM Length L Ch R = 1 ,32944   ,355.1,364.5,371
XS GIS Cut Line= 3
     2107205.495      184144.325       2107125.2       184840.94
     2106871.294      185233.735
#Sta/Elev= 30
       0 2352.72    48.8 2344.95   192.4 2328.88   223.8 2323.24   289.9  2306.2
   306.4 2299.91   322.9 2297.75   331.7 2295.37   355.9 2286.04   408.8  2268.1
   450.1 2252.19   468.2 2246.64     488 2237.72   531.2 2237.35   537.6 2235.96
   547.4 2237.34   613.5 2238.57   642.6 2241.44   696.1 2243.71   718.6 2246.39
   796.5 2259.69   834.6 2268.75   874.9 2280.23   923.4 2296.86   935.5 2298.88
   953.2 2305.24  1031.5 2328.64    1121 2352.66  1144.4  2359.8  1168.9 2365.49
#Mann= 5 ,-1 , 0
       0      .1       0     410     .04       0     510      .1       0
   531.2    .045       0   547.4      .1       0
#XS Ineff= 2 , 0
                          587.03         2241.08
Permanent Ineff=
       F       F
Bank Sta=531.2,547.4
XS Rating Curve= 0 ,0
Exp/Cntr=0.3,0.1

Type RM Length L Ch R = 1 ,32580   ,152.3,172,192.5
XS GIS Cut Line= 4
2107120.96560466184123.5400946322106885.96151873184495.230230534
2106790.04148366184655.8962892792106550.24139598185065.954439209
#Sta/Elev= 30
       0 2348.02    60.8 2335.09   109.1 2327.71     175 2315.84   217.8 2305.37
   258.2 2297.96     276  2293.5   336.7 2269.84   383.5 2248.94     408 2241.21
   438.8 2236.68   469.6 2230.61   500.2 2231.27   513.1 2229.93   528.4 2231.08
   589.7 2231.11   618.4 2233.39   643.8 2241.48   704.7 2249.18   733.5 2254.85
   759.3 2263.12   767.1 2264.21   793.3  2274.2   832.3  2285.7   880.9 2295.59
   910.3 2300.05   956.9 2304.17  1009.3 2303.69  1086.2 2297.55  1101.9 2293.95
#Mann= 4 ,-1 , 0
       0      .1       0     400     .04       0   500.2    .045       0
   528.4      .1       0
Bank Sta=500.2,528.4
XS Rating Curve= 0 ,0
Exp/Cntr(USF)=0,0
Exp/Cntr=0.5,0.3

Type RM Length L Ch R = 1 ,32408   ,60.6,61.5,54.7
XS GIS Cut Line= 4
     2106986.087      184031.531     2106720.245      184490.515
     2106674.672      184488.345     2106358.917      184949.499
#Sta/Elev= 30
       0 2347.79     8.9  2347.5    19.5 2344.59    38.5 2343.05      84 2335.46
   114.1 2333.96   144.7 2329.91   190.9 2317.43   231.7 2304.58   283.9 2294.28
     311 2284.47   391.1 2242.75   409.4 2235.05   421.3 2231.44     448 2228.64
   497.3 2229.08  544.382227.533   551.2  2226.2  564.772227.533   612.3 2229.37
   631.2 2233.62   659.5 2237.41   782.2 2249.79   790.4 2249.58   803.5 2247.33
   834.1 2256.16     866 2261.71   949.5 2279.74  1084.7 2314.95  1134.9 2326.28
#Mann= 5 ,-1 , 0
       0      .1       0     490     .04       0  544.38    .045       0
  564.77     .04       0  656.04      .1       0
#XS Ineff= 2 , 0
          494.19 2230.64  587.78         2230.64
Permanent Ineff=
       F       F
Bank Sta=544.38,564.77
XS Rating Curve= 0 ,0
Exp/Cntr=0.5,0.3
