HEC-RAS study DRPLKCR.prj: DRPLKCR

--- DRPLKCR.g01 (geometry) --- (continued)

Type RM Length L Ch R = 1 ,32346   ,168.6,148.2,134.3
XS GIS Cut Line= 4
     2106953.058       183987.13     2106687.216      184446.114
     2106641.643      184443.944     2106325.887      184905.098
#Sta/Elev= 30
       0  2349.7    36.7 2343.65   150.5  2331.6   211.4 2316.62   264.2 2301.87
   312.1 2291.76   335.8  2283.7   410.5 2242.49     431 2232.36   440.5 2229.13
   457.6 2227.93   491.7  2228.8   503.1 2226.84   531.3 2228.24   547.6 2227.87
  553.172226.609   560.9 2224.95  567.252226.611     574 2228.38     611 2227.59
   634.6 2229.78   671.1 2235.87   778.6 2244.94   788.6 2248.56   800.5 2249.82
   812.4 2254.42   864.1 2267.64  1007.5 2299.43  1090.1 2316.12  1134.9 2322.68
#Mann= 5 ,-1 , 0
       0      .1       0  550.41     .04       0  553.17    .045       0
  567.25     .04       0  696.04      .1       0
#XS Ineff= 2 , 0
          489.74 2229.37   598.7         2229.28
Permanent Ineff=
       F       F
Bank Sta=553.17,567.25
XS Rating Curve= 0 ,0
Exp/Cntr=0.5,0.3

Type RM Length L Ch R = 1 ,32198   ,364.5,369.6,365.4
XS GIS Cut Line= 2
     2106862.613      183933.822     2106202.891       184849.62
#Sta/Elev= 30
       0 2344.85    56.3 2334.14   133.2 2326.38   182.5 2318.84   211.8 2312.69
   262.4 2300.01   321.2 2288.41   356.5 2275.64     380 2265.91   408.2  2252.3
   438.7 2234.01   456.7 2226.27  466.952224.578   476.3 2223.34  482.992224.553
   582.2  2224.3   605.6  2226.8   631.5    2227   645.6 2229.39     709 2234.46
   731.6 2237.66   765.4 2244.88   784.2 2252.19   808.4 2259.88   820.6 2260.91
     861 2270.84   907.8 2278.42  1030.8 2290.51  1067.2 2291.73  1128.7    2291
#Mann= 5 ,-1 , 0
       0      .1       0  466.95    .045       0  482.99      .1       0
     520     .04       0     650      .1       0
Bank Sta=466.95,482.99
XS Rating Curve= 0 ,0
Exp/Cntr=0.3,0.1

Type RM Length L Ch R = 1 ,31829   ,312.4,310.4,305.2
XS GIS Cut Line= 2
     2106563.134      183734.169     2105914.263       184686.86
#Sta/Elev= 30
       0 2301.01    11.1 2299.54    38.3 2292.99      69  2288.2    95.9 2284.91
   139.9 2282.06   177.7 2275.62   200.8 2269.27   241.4 2256.02     281    2246
   304.8 2237.23   324.7 2231.92   356.4 2226.16   396.1 2221.45   432.7 2218.51
  486.952217.711   492.2 2217.14   503.3 2217.74   593.2 2218.36   645.2 2221.86
   689.9 2223.13     702  2224.4   795.2 2226.85   841.2 2230.74   895.5 2241.68
  1007.4 2268.72    1082 2283.36    1110 2286.87  1138.4 2288.56  1152.7 2287.98
#Mann= 9 ,-1 , 0
       0      .1       0  486.95    .045       0   503.3      .1       0
     640    .035       0     680     .06       0     760     .04       0
     850    .035       0     870     .08       0    1110      .1       0
Bank Sta=486.95,503.3
XS Rating Curve= 0 ,0
Exp/Cntr=0.3,0.1

Type RM Length L Ch R = 1 ,31518   ,426,448.4,416.5
XS GIS Cut Line= 3
     2106530.582      183708.127     2106239.784       183755.87
     2105860.009      184630.436
#Sta/Elev= 30
       0 2295.63    54.9 2282.14   114.6 2269.75   164.7 2256.28   174.6 2251.53
     214 2224.96   227.8 2218.72   267.7 2217.92   287.7 2215.26   294.3 2217.09
   313.2 2216.19   334.7  2216.8   376.2 2213.57   409.1 2214.57   449.1 2213.74
  453.822212.778   459.9 2211.56   466.9 2212.89   474.2 2213.48   509.9 2212.07
   681.4 2214.68     739 2214.48   799.6 2221.03   821.1 2220.54   831.8 2224.24
   867.6 2227.55   974.9 2249.86  1077.9 2267.61    1211 2294.08  1248.2 2299.85
#Mann= 10 ,-1 , 0
       0      .1       0     260    .035       0  304.69      .1       0
  453.82    .045       0   466.9      .1       0  684.69    .035       0
  734.69     .04       0  844.69     .06       0  934.69     .08       0
 1174.69      .1       0
#XS Ineff= 2 , 0
             409 2215.61  634.39         2215.11
Permanent Ineff=
       F       F
Bank Sta=453.82,466.9
XS Rating Curve= 0 ,0
Exp/Cntr=0.3,0.1

Type RM Length L Ch R = 1 ,31070   ,211.8,226.4,197.3
XS GIS Cut Line= 2
     2106107.405      183397.798     2105640.825      184456.825
#Sta/Elev= 30
       0 2252.66    62.1  2243.6   108.7 2235.89     123 2230.69   137.4 2231.42
   148.1 2229.43   223.4 2223.07   427.9 2210.83   463.6 2209.29     478 2207.82
  516.242206.906   527.2 2205.42  538.222206.906   696.5 2208.14   750.4 2210.48
   775.5 2210.07   786.3 2212.06   800.6 2213.22   803.5 2214.01     815 2220.99
   836.5 2230.08   843.6 2233.89   861.6  2240.1   883.2 2245.97   933.3 2257.54
   954.8  2263.4   997.2 2273.43  1043.2 2285.67  1094.7 2300.37  1157.3 2319.88
#Mann= 9 ,-1 , 0
       0      .1       0     190     .04       0     300    .035       0
     510      .1       0  516.24    .045       0  538.22      .1       0
     550    .035       0     730     .06       0     790      .1       0
#XS Ineff= 2 ,-1
       0  506.52 2209.48  643.32  1157.2 2209.39
Permanent Ineff=
       F       F
Bank Sta=516.24,538.22
XS Rating Curve= 0 ,0
Exp/Cntr=0.5,0.3

Type RM Length L Ch R = 1 ,30843   ,40.3,45.1,48.6
XS GIS Cut Line= 4
2106075.77508504183389.114509762 2105740.1841426183762.937331727
2105750.09611136183937.1047828692105595.75259775184425.623243391
#Sta/Elev= 30
       0 2257.75    60.1 2251.45   176.2 2235.73   198.2 2230.41   202.6 2229.97
   220.3 2231.16   237.9 2228.23   254.9  2226.6   365.8 2219.06   397.3 2217.75
     471 2210.98   495.5  2207.9   522.1 2205.97   550.3 2205.89   568.2 2204.66
   584.7 2205.22   621.62203.257   627.3 2201.94   643.7 2202.16  648.32 2203.27
   653.6 2204.96   782.9 2206.81   838.3 2212.67   855.5 2219.13   872.7 2227.55
   944.9 2253.93   971.1 2261.95  1075.8 2290.43  1161.2  2315.7  1189.1 2324.69
#Mann= 8 ,-1 , 0
       0      .1       0     240     .04       0     380    .035       0
     430     .04       0  602.36     .06       0   621.6    .045       0
  648.32     .06       0  806.81      .1       0
#XS Ineff= 3 ,-1
       0  618.14  2203.3  652.45  720.17 2203.47   728.2  804.53 2207.11
Permanent Ineff=
       F       F       F
Bank Sta=621.6,648.32
XS Rating Curve= 0 ,0
Exp/Cntr(USF)=0,0
Exp/Cntr=0.5,0.3

Type RM Length L Ch R = 1 ,30798   ,124.2,142.7,158.9
XS GIS Cut Line= 4
2105903.02362944183321.1467239512105711.86423184183731.785429897
2105711.86423184183965.4246936242105574.51266468184411.463288014
#Sta/Elev= 30
       0 2290.73    48.6 2287.53    78.5 2282.96   129.1 2270.57     187 2258.37
   212.8 2248.66   258.4 2238.62   277.5 2236.05   295.6 2229.94   317.3 2230.85
   335.4  2227.1   365.3 2224.21   389.7 2219.36   407.8 2218.33   429.5 2212.01
   474.4 2207.25   582.7 2202.74   589.2 2201.37   595.7 2201.48  600.42 2202.79
   605.5  2203.7     746 2206.43   800.2 2213.06   814.6 2217.76   824.9 2223.05
     842 2228.68   862.7 2237.03   931.2  2261.2  1041.7    2292  1153.3 2326.27
#Mann= 6 ,-1 , 0
       0      .1       0     280     .04       0   582.7    .045       0
  600.42     .06       0  756.59     .04       0  786.59      .1       0
#XS Ineff= 2 , 0
          579.39 2202.84  667.05         2210.51
Permanent Ineff=
       F       F
Bank Sta=582.7,600.42
XS Rating Curve= 0 ,0
Exp/Cntr(USF)=0,0
Exp/Cntr=0.5,0.3

Type RM Length L Ch R = 1 ,30656   ,207.8,201.7,190.8
XS GIS Cut Line= 4
2105881.40866594  183300.50647972105647.71501206183759.547585537
2105488.37842986183887.7755969192105332.07683019184266.389666031
#Sta/Elev= 30
       0 2295.49    44.1 2293.57    84.3 2288.39     195 2266.38   277.2  2245.3
   327.5 2236.46   353.3 2229.51   408.5 2229.52   441.7 2221.05     465  2209.2
   479.7  2204.1   493.2 2202.96   515.1 2203.77   558.2 2200.05   576.32200.238
   586.2 2198.72   592.82200.852   609.6 2203.97   703.8 2204.83   714.8 2212.84
     719 2214.74   751.9 2223.01   769.5 2228.58   778.6 2233.25   789.5 2237.01
     865 2260.83   921.8 2276.08   962.9 2288.51  1067.4 2323.38  1129.2 2345.44
#Mann= 7 ,-1 , 0
       0      .1       0     300     .04       0     420      .1       0
   576.3    .045       0   592.8      .1       0   685.1     .04       0
  799.63      .1       0
Bank Sta=576.3,592.8
XS Rating Curve= 0 ,0
Exp/Cntr(USF)=0,0
Exp/Cntr=0.3,0.1

Type RM Length L Ch R = 1 ,30454   ,123.4,121.4,121.7
XS GIS Cut Line= 3
     2105735.924      183194.184     2105469.921      183660.816
     2105234.854      184214.898
#Sta/Elev= 30
       0 2317.09    99.6 2305.21   110.9 2302.32   122.3 2301.57   201.6  2287.2
     228 2281.36   235.6 2280.44   357.6 2248.22   416.8 2235.56   432.2 2234.14
   443.3 2231.62   454.6 2230.42   466.1 2226.95   511.6 2200.11  526.182195.287
   530.8 2193.98   537.7 2193.67  546.742195.287   551.9 2196.79   635.7 2199.57
   680.7 2206.57   700.7 2207.22   712.3  2214.4   740.8  2224.3   810.8 2245.23
   875.9  2261.3   936.8 2279.44   954.6 2286.19   997.4 2300.12    1139 2352.25
#Mann= 5 ,-1 , 0
       0      .1       0  526.18    .045       0  546.74      .1       0
  657.12     .04       0  757.12      .1       0
#XS Ineff= 2 , 0
                           558.1         2202.21
Permanent Ineff=
       F       F
Bank Sta=526.18,546.74
XS Rating Curve= 0 ,0
Exp/Cntr=0.3,0.1

Type RM Length L Ch R = 1 ,30333   ,152.9,151,150
XS GIS Cut Line= 2
2105572.50344083183123.4866488872105114.54997448184175.738818169
#Sta/Elev= 30
       0 2320.39    99.9 2306.64   146.4 2294.97   160.7 2293.33   199.1 2282.33
   303.9 2247.62   343.2    2236     379  2226.7   434.9 2216.73   457.7 2210.59
   482.8 2201.48   508.32194.089   514.6  2191.8   522.1 2191.62   527.22193.333
   536.4 2196.25   543.6 2193.98     552 2193.94   565.1 2197.95   631.8 2200.84
   646.8 2205.13   658.1 2210.73   676.7 2211.65   694.1 2222.17   711.6 2229.14
   733.2 2234.82   785.2 2245.45     812 2253.09  1015.7 2324.38  1147.6 2365.77
#Mann= 7 ,-1 , 0
       0      .1       0     440     .06       0     490      .1       0
   508.3    .045       0   527.2      .1       0     600     .04       0
     700      .1       0
Bank Sta=508.3,527.2
XS Rating Curve= 0 ,0
Exp/Cntr(USF)=0,0
Exp/Cntr=0.3,0.1

Type RM Length L Ch R = 1 ,30182   ,156.9,146.1,133.4
XS GIS Cut Line= 2
      2105406.45      183052.745     2105000.634      184168.197
#Sta/Elev= 30
       0 2336.82    99.5 2319.94   179.8 2298.71   207.7 2288.08   221.6 2285.67
   244.2 2277.89   332.5  2244.5   389.2 2227.06   427.6 2217.55   459.2 2203.89
   479.7 2197.57  491.212191.585   500.1  2190.7   507.8 2191.79   521.9 2194.14
   535.9 2190.75   556.8 2190.02   595.2 2196.75   612.7  2197.8   633.6 2201.38
   651.1 2205.75   682.5 2216.36   713.9 2215.47   738.3 2228.84   774.1 2240.08
   867.5 2277.22   982.7 2319.74  1045.9 2338.58  1136.3 2362.91    1187 2373.29
#Mann= 5 ,-1 , 0
       0      .1       0  491.21    .045       0   507.8      .1       0
     660     .04       0     760      .1       0
#XS Ineff= 2 , 0
                           519.2         2203.53
Permanent Ineff=
       F       F
Bank Sta=491.21,507.8
XS Rating Curve= 0 ,0
Exp/Cntr=0.3,0.1

Type RM Length L Ch R = 1 ,30036   ,249.7,269.6,294.1
XS GIS Cut Line= 4
2105200.70977453183035.011669811 2105088.4833335183475.284630789
2105123.01454613183585.3528710332104961.14948694184155.117879358
#Sta/Elev= 30
       0 2340.22   129.7 2310.58   260.3 2271.16     284 2261.66     301 2258.43
   311.1 2253.85   324.7 2249.66   365.3 2238.14   412.7 2229.09   443.2 2217.29
   467.1 2206.01   484.8 2191.29   491.1 2188.71   511.8 2191.35   525.5 2193.45
   539.3 2189.15   545.2  2188.5   583.9 2188.93   600.9 2193.94   628.2 2195.82
   679.4 2204.24     691 2207.04   713.5 2215.04   737.3 2216.17   757.8  2230.1
   863.5 2280.86   935.3 2310.02   962.4  2319.2  1054.5 2345.84    1162 2369.22
#Mann= 5 ,-1 , 0
       0      .1       0   484.8    .045       0   511.8      .1       0
  759.71     .04       0  859.71      .1       0
#XS Ineff= 2 , 0
                          520.92         2202.43
Permanent Ineff=
       F       F
Bank Sta=484.8,511.8
XS Rating Curve= 0 ,0
Exp/Cntr(USF)=0,0
Exp/Cntr=0.5,0.3

Type RM Length L Ch R = 1 ,29766   ,34.2,46.5,45.9
XS GIS Cut Line= 4
     2105049.813      182998.034     2104937.834      183664.701
     2104898.772       183676.42     2104867.522      184155.587
#Sta/Elev= 30
       0 2344.13   146.9 2312.35   243.4 2284.18   349.9 2256.35   363.2 2251.38
   393.1 2248.03   476.3 2227.25   499.7 2216.92   512.9 2214.73   532.8 2207.12
   549.5  2195.8   592.7 2187.01   645.9 2186.84   656.1 2189.03   665.9 2188.39
  673.832185.604     687 2184.96  697.322185.604   703.6 2188.34   718.1 2188.67
     751 2194.86   777.1 2207.67   793.7 2212.42   816.7 2213.27   836.4 2227.07
   960.3 2283.14    1014 2306.35  1056.7 2321.59  1086.9 2330.48    1197 2350.88
#Mann= 5 ,-1 , 0
       0      .1       0  673.83    .045       0  697.32      .1       0
  806.79     .04       0  906.79      .1       0
#XS Ineff= 2 , 0
          662.93 2192.33  704.73         2192.27
Permanent Ineff=
       F       F
Bank Sta=673.83,697.32
XS Rating Curve= 0 ,0
Exp/Cntr=0.5,0.3

Type RM Length L Ch R = 1 ,29719   ,160.1,141.3,122.8
XS GIS Cut Line= 4
      2105027.07      182974.944     2104917.695      183624.684
     2104878.633      183636.403     2104846.081      184144.215
#Sta/Elev= 30
       0 2347.85    32.6 2342.03    40.6 2338.91    57.2 2337.28   149.4 2316.37
   359.8 2257.33   443.2 2239.49     503 2220.78   519.6 2217.97   546.3 2207.52
   569.6    2202   606.2  2186.5   649.4 2186.23  670.78 2182.57   679.1 2181.38
  684.222182.571   692.8 2185.11     741 2188.08   767.3 2193.98   794.2 2204.52
   810.1 2206.85     820 2211.89     843 2211.89   862.7 2225.14   957.9 2267.19
  1046.8 2303.42  1125.7 2327.62  1132.3 2331.35  1155.3 2332.62  1208.5 2343.27
#Mann= 5 ,-1 , 0
       0      .1       0  670.78    .045       0  684.22      .1       0
  829.66     .04       0  929.66      .1       0
#XS Ineff= 2 , 0
          660.23 2189.44   687.9         2189.28
Permanent Ineff=
       F       F
Bank Sta=670.78,684.22
XS Rating Curve= 0 ,0
Exp/Cntr=0.5,0.3

Type RM Length L Ch R = 1 ,29578   ,169.2,169.6,165.6
XS GIS Cut Line= 4
2104894.24526248182985.3730516612104820.86643565183438.595217374
2104758.27861277183680.3137057542104741.01300645184129.219469888
#Sta/Elev= 30
       0 2345.17      10 2341.62    26.7 2340.03    89.8 2325.07   254.8 2272.32
   322.5 2253.38   332.4 2249.17   345.7 2247.86     379  2241.5   415.5 2225.86
   452.1 2212.45   473.3 2205.88   526.5 2193.34   535.3 2188.98   543.4 2181.37
  549.362179.065   560.4 2177.82  568.652179.065   577.3  2182.1     696 2186.28
   735.8 2190.36   788.3 2202.02   804.7 2207.25   827.7 2207.74   844.1  2218.8
   909.7 2245.77  1036.1  2291.3  1087.4 2307.51  1129.7 2317.09  1158.1 2321.17
#Mann= 5 ,-1 , 0
       0      .1       0  549.36    .045       0  568.65      .1       0
  798.81     .04       0  898.81      .1       0
#XS Ineff= 2 , 0
                          625.79         2193.11
Permanent Ineff=
       F       F
Bank Sta=549.36,568.65
XS Rating Curve= 0 ,0
Exp/Cntr(USF)=0,0
Exp/Cntr=0.3,0.1

Type RM Length L Ch R = 1 ,29409   ,152.3,143.3,138.3
XS GIS Cut Line= 3
     2104767.335      182964.988     2104640.285      183473.197
     2104645.197      184144.697
#Sta/Elev= 30
       0 2346.51    41.4  2337.4    54.9 2336.22   132.7 2311.13   184.8  2292.2
   196.9 2289.64   264.6 2266.42   274.1 2261.59   287.7 2260.23   433.5 2210.66
   494.5 2193.25   501.3 2189.03   508.1 2180.09  513.992176.348   524.9 2175.25
  530.322176.347   541.3 2182.44   547.9 2183.16   603.7 2183.36   648.4 2179.54
   705.4 2179.43   715.2 2181.97   764.1 2187.06   836.6 2192.43   856.3 2201.67
   879.3 2201.16   895.7 2210.32  1070.9 2270.98    1131 2284.96  1195.4 2294.12
#Mann= 6 ,-1 , 0
       0      .1       0  513.99    .045       0  530.32     .06       0
  623.85      .1       0  823.85     .04       0  913.85      .1       0
#XS Ineff= 2 , 0
                          572.98         2186.42
Permanent Ineff=
       F       F
Bank Sta=513.99,530.32
XS Rating Curve= 0 ,0
Exp/Cntr=0.3,0.1

Type RM Length L Ch R = 1 ,29265   ,211.6,202.6,193.9
XS GIS Cut Line= 5
2104421.59928967182983.2148508722104475.55430939183371.690992912
2104512.24372281183518.4486465712104607.20455753183829.229560202
2104617.99556148184144.326875412
#Sta/Elev= 30
       0 2291.88      61 2301.62   108.2 2303.19   151.2 2298.38   333.5 2268.21
   353.4 2261.58   379.9 2248.99   406.7 2234.06   437.1 2210.16   447.2 2200.42
   464.1 2180.79  477.342174.445   487.2 2173.15  495.172174.444   511.5 2179.94
   528.4 2181.33   618.3 2181.33   703.1  2179.1     812 2189.02   833.5  2189.2
   840.4 2191.43   848.8 2197.86   854.1 2199.73   877.7 2198.61   894.1 2208.58
     963 2230.15  1012.3 2247.99  1077.9 2267.64    1137 2280.55  1183.7 2286.69
#Mann= 7 ,-1 , 0
       0      .1       0  477.34    .045       0  495.17      .1       0
  603.48    .025       0  703.48      .1       0  803.48     .06       0
  908.44      .1       0
#XS Ineff= 2 , 0
                          557.02         2188.61
Permanent Ineff=
       F       F
Bank Sta=477.34,495.17
XS Rating Curve= 0 ,0
Exp/Cntr(USF)=0,0
Exp/Cntr=0.3,0.1

Type RM Length L Ch R = 1 ,29063   ,225.2,229.8,236.7
XS GIS Cut Line= 3
     2103971.988      183150.402     2104403.846      183634.343
     2104555.878      184161.728
#Sta/Elev= 30
       0 2204.01    65.2 2198.82   129.8  2200.2   155.8 2194.16   216.2 2195.44
   304.5  2243.3   315.4 2244.84   336.7 2252.12   381.1 2251.39   420.5 2245.07
   446.3 2233.53   464.9 2222.36   500.1 2196.06   504.4 2191.95   514.1 2177.84
  519.382172.124   526.4 2170.66  536.182172.123   548.4 2175.89   561.6 2176.37
   574.1 2180.73     588 2178.74   814.2 2178.71   847.4 2180.77   881.5 2190.17
   917.5 2189.56   960.1 2212.96   997.6  2225.5  1144.4 2262.33  1197.5 2272.64
#Mann= 8 ,-1 , 0
       0      .1       0      40    .035       0     170     .04       0
     300      .1       0  519.38    .045       0  536.18      .1       0
  788.61     .06       0  998.61      .1       0
#XS Ineff= 2 , 0
                          546.13         2179.05
Permanent Ineff=
       F       F
Bank Sta=519.38,536.18
XS Rating Curve= 0 ,0
Exp/Cntr=0.3,0.1

Type RM Length L Ch R = 1 ,28833   ,137.1,143.5,142.2
XS GIS Cut Line= 4
2103938.16231291183151.5545124232104115.13477761183598.302075768
2104281.31623837183952.2470051812104402.17548256184239.287710133
#Sta/Elev= 30
       0 2205.71    54.2  2200.1   160.1 2193.27   181.3 2189.36   227.2 2190.32
   244.8 2188.85     266 2191.24   276.6  2198.6     333 2226.84   348.8 2227.75
   368.3 2234.12     393 2235.85   422.2 2232.33   442.3 2227.33   463.6 2218.39
     532 2184.59   575.5 2176.17   593.6 2175.73   603.6 2169.47   609.5 2168.75
   620.6 2169.41   803.8 2170.22   925.1 2179.06   943.9 2184.11     965  2192.5
   985.2 2194.21  1005.2 2206.05  1015.7 2209.13  1068.5 2217.84    1183 2241.57
#Mann= 8 ,-1 , 0
       0      .1       0      30    .035       0     230     .04       0
     350      .1       0   603.6    .045       0   620.6      .1       0
  881.54     .04       0 1101.54      .1       0
Bank Sta=603.6,620.6
XS Rating Curve= 0 ,0
Exp/Cntr(USF)=0,0
Exp/Cntr=0.5,0.3

Type RM Length L Ch R = 1 ,28689   ,31.6,29.5,28.9
XS GIS Cut Line= 2
     2103895.733       183162.01     2104255.108      184339.093
#Sta/Elev= 30
       0 2208.13    79.5 2198.54   182.4 2191.53   212.2  2187.4   233.9 2187.47
   257.9 2184.97   283.2 2185.34   301.6 2188.58   322.6 2188.11   347.1 2196.05
   367.7  2199.1   453.4 2203.74   467.2 2201.86   501.5 2193.58   549.5 2178.56
   622.2 2172.67  701.392168.306   710.7 2166.96   716.8 2168.41   798.3  2168.4
   815.5 2170.62   871.6 2174.16   889.1 2174.11   899.4 2172.26   933.7 2177.01
     992 2178.09  1022.9 2181.64  1166.9 2189.35    1191 2189.63  1230.7 2199.57
#Mann= 12 ,-1 , 0
       0      .1       0      20    .035       0     220     .04       0
     430      .1       0     530     .04       0  701.39    .045       0
   716.8     .04       0     770      .1       0     840     .04       0
     940      .1       0    1100     .04       0    1150      .1       0
#XS Ineff= 2 , 0
          691.98 2175.01  730.09          2174.9
Permanent Ineff=
       F       F
Bank Sta=701.39,716.8
XS Rating Curve= 0 ,0
Exp/Cntr=0.5,0.3

Type RM Length L Ch R = 1 ,28660   ,294.1,301.3,307.2
XS GIS Cut Line= 2
     2103870.994      183175.031     2104230.369      184352.114
#Sta/Elev= 30
       0 2209.69    92.9 2197.24   181.1 2191.46   268.3 2182.85   288.9 2184.14
   327.2 2182.81   349.6 2185.94   394.6 2185.57   450.8 2190.16   477.6 2188.18
   522.1 2178.68   583.9  2172.8   664.2 2171.96   700.5  2168.4  707.092165.827
   713.1 2164.74  720.812165.828   728.8 2169.46   806.9 2169.33   833.9 2172.95
   889.2 2173.15   950.9 2176.99   971.5 2179.38   995.5 2187.31    1035 2192.89
  1074.4 2191.94  1098.4  2186.4  1180.6 2191.98  1207.1 2190.96  1230.7 2194.49
#Mann= 9 ,-1 , 0
       0    .035       0     210     .04       0     510      .1       0
     520     .04       0  707.09    .045       0  720.81     .04       0
     830     .06       0     850     .04       0     930      .1       0
#XS Ineff= 2 , 0
           700.5 2171.65  726.25         2171.55
Permanent Ineff=
       F       F
Bank Sta=707.09,720.81
XS Rating Curve= 0 ,0
Exp/Cntr=0.5,0.3

Type RM Length L Ch R = 1 ,28359   ,233.8,239.5,242.8
XS GIS Cut Line= 3
     2103845.088      183165.716      2103791.59      183882.293
     2103725.335      184405.816
#Sta/Elev= 30
       0 2218.89     6.8 2217.84    32.2 2210.72    56.1  2205.3   230.5 2190.42
   263.4 2189.19   302.9 2186.04   355.5 2184.26   457.5 2178.47   590.4 2174.16
   673.6 2169.01   687.8 2169.66   704.2 2165.73  711.062160.816   714.1 2159.44
   717.4 2159.23  725.192160.817   733.6 2162.13   902.6 2162.13   922.9  2162.8
   935.6 2165.06   945.5 2165.82   962.1 2165.99  1047.8 2210.93  1128.3 2248.55
    1144 2256.59    1169  2266.6  1203.5 2282.07  1239.9 2296.83  1246.3 2298.67
#Mann= 8 ,-1 , 0
       0      .1       0      10    .035       0     610      .1       0
  711.06    .045       0  725.19      .1       0  798.57    .035       0
  998.57     .04       0 1098.57      .1       0
#XS Ineff= 2 , 0
                          798.13          2165.8
Permanent Ineff=
       F       F
Bank Sta=711.06,725.19
XS Rating Curve= 0 ,0
Exp/Cntr=0.3,0.1

Type RM Length L Ch R = 1 ,28119   ,150.9,163.5,168.1
XS GIS Cut Line= 5
2103793.85771549183186.642444306 2103536.8692383183934.478912933
2103452.06304083183940.9036248632103421.22442357183982.021781214
  2103326.138687184236.440373633
#Sta/Elev= 30
       0  2234.6   104.7 2208.95   120.3 2207.54   144.6 2203.26   359.7 2187.38
   505.4 2179.17   602.5 2169.39   668.4 2166.17   682.3 2167.08   703.1  2164.9
   720.4    2157   737.8 2156.25   746.3 2156.91   751.7 2158.31   772.1 2158.15
   795.4 2160.45   873.1 2160.44   899.5 2159.41   945.6 2160.72   984.1 2163.53
  1001.2 2163.81  1011.4 2170.02  1029.3 2178.09  1067.5 2197.68  1087.9 2206.03
  1103.2  2210.2  1124.2 2214.03  1145.2 2215.65  1176.7 2215.51  1198.8 2213.98
#Mann= 10 ,-1 , 0
       0      .1       0     220    .035       0     300      .1       0
     410    .035       0     720      .1       0   720.4    .045       0
   746.3      .1       0  905.81     .06       0  915.81     .04       0
 1017.21      .1       0
Bank Sta=720.4,746.3
XS Rating Curve= 0 ,0
Exp/Cntr(USF)=0,0
Exp/Cntr=0.3,0.1

Type RM Length L Ch R = 1 ,27956   ,549.5,567.5,566.7
XS GIS Cut Line= 3
     2103733.273      183176.443     2103511.919      183766.721
     2103175.547      184202.919
#Sta/Elev= 30
       0 2258.63    69.3 2240.04   121.9 2221.56   149.9 2213.24   177.9 2207.18
   205.6 2203.43   311.1 2192.68   361.1 2190.19   381.2 2187.64   475.8  2181.5
   562.4 2167.71   642.3 2162.64   722.4 2160.68   736.4 2159.54     750 2155.96
   803.9 2154.75   812.2 2153.98   820.4 2154.71   826.2 2156.13   890.6  2161.2
   907.1    2164   932.9 2164.63   942.2  2166.7     961 2167.46     975 2172.09
   986.7 2171.25  1051.8 2174.01  1067.9 2175.99  1102.2 2186.92  1181.2  2220.8
#Mann= 9 ,-1 , 0
       0      .1       0     210    .035       0     310      .1       0
     420    .035       0     630      .1       0   803.9    .045       0
   820.4      .1       0  880.42     .04       0 1000.42      .1       0
#XS Ineff= 2 , 0
                          830.65          2159.1
Permanent Ineff=
       F       F
Bank Sta=803.9,820.4
XS Rating Curve= 0 ,0
Exp/Cntr=0.3,0.1

Type RM Length L Ch R = 1 ,27388   ,442.4,429.5,416.5
XS GIS Cut Line= 3
     2103585.704      183111.339     2103425.113      183337.034
     2102708.968       183742.85
#Sta/Elev= 30
       0 2277.31    48.4 2261.91    99.2 2238.88   131.4 2228.18   194.2 2214.07
   268.3 2195.47   295.9 2186.92   333.5 2171.98   344.8 2165.56   363.6 2151.87
   371.2 2148.67   384.9 2146.86     424 2147.97   435.3 2146.42     473 2147.89
  480.94 2145.75   488.1 2144.53  496.762145.749   505.2 2147.83   574.8 2147.65
   589.9 2150.59     622 2153.08     847  2179.7   865.2 2181.96   887.9 2181.05
   897.6 2184.39   925.5 2187.91     957 2196.95  1034.5 2226.16  1100.1 2249.17
#Mann= 5 ,-1 , 0
       0      .1       0  480.94    .045       0  496.76      .1       0
     847     .04       0     957      .1       0
Bank Sta=480.94,496.76
XS Rating Curve= 0 ,0
Exp/Cntr=0.3,0.1

Type RM Length L Ch R = 1 ,26959   ,406.7,400.4,381.6
XS GIS Cut Line= 3
     2103053.077      182679.886     2102942.914      183207.495
      2102645.05      183712.193
#Sta/Elev= 30
       0 2290.66    23.9 2288.72    47.4 2284.41    79.6    2275   151.7 2259.13
   184.8 2249.15   208.3    2240   245.1  2217.9   302.1 2187.68   325.6 2172.36
     349 2152.76     368  2142.4   385.9 2141.17   459.6  2141.8  529.322140.469
   536.7 2138.71  546.262140.467   559.3 2141.87   575.7 2145.94   700.3 2152.26
   783.6 2161.22   837.4 2164.38   883.1 2170.62   902.1 2176.95   921.2 2176.46
     925 2177.43   936.4 2184.14  1020.2 2216.26  1069.7 2233.47    1125 2249.37
#Mann= 7 ,-1 , 0
       0      .1       0  529.32    .045       0  546.26      .1       0
  618.99    .035       0  748.99      .1       0  848.99     .04       0
  958.99      .1       0
Bank Sta=529.32,546.26
XS Rating Curve= 0 ,0
Exp/Cntr=0.3,0.1

Type RM Length L Ch R = 1 ,26558   ,292.6,299.6,302.1
XS GIS Cut Line= 4
2102601.29039263182628.3371145222102569.56342014183042.374105552
2102679.02147524183416.7523809662102561.63167701183699.122436151
#Sta/Elev= 30
       0 2209.49    48.9 2196.13    75.2 2186.98    85.1  2180.9      97 2179.49
   124.5 2173.74   213.4 2160.05   256.2 2157.38     285 2151.16     322 2150.67
     342 2149.12   404.2 2142.09   427.7 2137.93     438 2137.35   441.92135.208
   448.2 2133.86   460.6 2135.27   475.6 2137.01   543.9 2136.52     591  2137.7
   660.2 2141.64   823.4 2166.64   845.7 2170.68   853.4 2173.75   878.3 2172.51
   890.9 2179.75     992 2201.03  1011.4 2206.28    1063 2223.16  1111.1 2235.86
#Mann= 8 ,-1 , 0
       0      .1       0     260    .035       0     350      .1       0
   441.9    .045       0   460.6    .035       0  555.25      .1       0
  765.25     .04       0   905.3      .1       0
Bank Sta=441.9,460.6
XS Rating Curve= 0 ,0
Exp/Cntr(USF)=0,0
Exp/Cntr=0.3,0.1

Type RM Length L Ch R = 1 ,26259   ,342,350,360.8
XS GIS Cut Line= 3
     2102312.684      182564.633     2102287.944      183127.601
     2102365.503      183667.464
#Sta/Elev= 30
       0 2246.97      14 2243.05    66.5 2224.36   102.7 2213.97   188.1 2184.13
   240.6 2169.36     303 2146.41   330.8 2143.22   391.7 2139.16   539.4 2137.57
     546 2136.19  551.312132.369   557.7 2130.79   565.7 2130.86   573.1 2132.17
   598.9 2131.34   629.5 2132.32   668.5 2131.59   681.7 2132.77   767.9 2132.94
   801.1 2136.76   807.7 2139.31     821 2147.74     831 2149.23   847.5 2150.11
   869.4 2166.61   887.2 2177.05   961.4    2217  1023.1 2246.53  1108.9 2283.25
#Mann= 5 ,-1 , 0
       0      .1       0  551.31    .045       0   573.1      .1       0
  813.51     .04       0  913.51      .1       0
Bank Sta=551.31,573.1
XS Rating Curve= 0 ,0
Exp/Cntr=0.3,0.1

Type RM Length L Ch R = 1 ,25909   ,345,350,347.3
XS GIS Cut Line= 3
      2102176.75      182524.053     2101977.159      183031.255
     2101737.603      183529.964
#Sta/Elev= 30
       0  2240.8    38.2 2224.97    68.6 2214.36   125.6 2190.18   186.9 2168.83
   245.5 2149.84   368.9 2133.93   397.1 2132.49   421.8 2132.86   527.6 2130.52
  536.152127.263   541.7 2126.25  550.21 2127.26   556.1 2128.77   603.9 2127.77
   719.9  2128.1   745.9 2129.44   756.3  2133.7   763.6 2135.31   785.4 2135.54
   789.1 2136.87   803.6 2148.46   821.8 2159.87   858.2 2184.95   887.3 2200.89
   905.5  2208.9     945  2220.4   992.9 2231.87  1054.8 2243.44  1098.3 2249.06
#Mann= 7 ,-1 , 0
       0      .1       0  536.15    .045       0  550.21      .1       0
  595.06     .07       0  705.06      .1       0  815.06     .04       0
  925.06      .1       0
#XS Ineff= 2 , 0
          524.81 2132.97  642.39         2132.33
Permanent Ineff=
       F       F
Bank Sta=536.15,550.21
XS Rating Curve= 0 ,0
Exp/Cntr=0.3,0.1

Type RM Length L Ch R = 1 ,25559   ,138.2,136.2,137.4
XS GIS Cut Line= 3
     2101920.306      182407.134     2101664.617      182888.374
     2101457.705      183399.362
#Sta/Elev= 30
       0 2240.09    30.7  2232.3    56.7 2223.56     121 2193.03   138.5 2185.93
     164 2178.22   268.5 2157.38   305.6  2151.5   324.1 2147.83   335.4 2144.32
   389.6 2141.01   417.1  2137.6   439.4 2132.64   461.7 2130.37   476.5 2130.21
   502.6 2124.41  529.812122.548   539.7 2120.74  553.212122.548   562.5  2125.6
   571.8 2126.48     678 2127.32   752.3 2129.79   773.6  2128.6   789.2 2137.27
   854.7 2168.75   890.4 2182.27   957.6 2211.22  1014.3 2232.12  1096.2 2256.66
#Mann= 7 ,-1 , 0
       0      .1       0     430     .07       0  529.81    .045       0
  553.21     .07       0  564.95    .025       0  644.95     .04       0
  834.95      .1       0
#XS Ineff= 2 , 0
                           576.1         2130.14
Permanent Ineff=
       F       F
Bank Sta=529.81,553.21
XS Rating Curve= 0 ,0
Exp/Cntr=0.3,0.1

Type RM Length L Ch R = 1 ,25422   ,155.1,154.8,153.7
XS GIS Cut Line= 4
2101746.85060672182365.4819216442101564.26681996182785.036155047
2101453.55111948183025.8913631122101338.95065757183379.404652368
#Sta/Elev= 30
       0 2233.76    14.2 2230.99    50.9 2219.78   125.7 2193.72   164.5 2181.56
   218.1  2167.3   253.9  2159.1   271.8 2156.92   325.1 2146.42   381.8  2137.8
     440 2129.49   457.9 2128.98   479.5 2123.02  511.822121.787     524 2120.38
  533.452121.788   537.3 2123.65   541.4 2124.11   555.4 2121.96     670 2121.98
   692.6 2124.75   738.8 2123.61     756 2125.29   787.1  2139.2   880.2 2188.39
   969.3 2240.88   980.2 2245.68  1035.4 2274.85  1076.8 2294.26  1094.3 2301.37
#Mann= 6 ,-1 , 0
       0      .1       0  477.56     .07       0  511.82    .045       0
  533.45     .07       0  567.56     .04       0  707.56      .1       0
#XS Ineff= 2 , 0
                           689.4         2140.29
Permanent Ineff=
       F       F
Bank Sta=511.82,533.45
XS Rating Curve= 0 ,0
Exp/Cntr(USF)=0,0
Exp/Cntr=0.3,0.1

Type RM Length L Ch R = 1 ,25268   ,206.7,180.4,151.3
XS GIS Cut Line= 4
2101560.38205854 182326.634307442101414.70350527182740.361398713
 2101381.6830332182819.9990078312101232.11971851183375.519890948
#Sta/Elev= 30
       0 2228.91    65.3 2213.92   145.4 2192.97   166.3 2186.76   194.1 2176.31
   206.9 2173.86   235.9 2165.55   270.6 2153.75   289.2 2153.39   315.9 2147.17
   368.9  2143.5   433.2 2129.65   448.2 2127.87   462.4 2127.87   480.2 2121.55
   483.7 2119.91   490.8  2119.1   497.9 2119.19   505.1 2121.28   515.7 2122.79
   550.1 2121.82   641.5 2122.55   662.2 2120.44   736.9 2121.17   745.9 2123.07
   780.7 2140.43   818.1 2164.24     900 2212.14  1039.3 2284.33  1100.1 2314.15
#Mann= 7 ,-1 , 0
       0      .1       0     380     .07       0   480.2    .045       0
   505.1     .07       0  594.84     .06       0  604.84     .04       0
  694.84      .1       0
#XS Ineff= 2 , 0
                          632.66         2141.39
Permanent Ineff=
       F       F
Bank Sta=480.2,505.1
XS Rating Curve= 0 ,0
Exp/Cntr(USF)=0,0
Exp/Cntr=0.5,0.3

Type RM Length L Ch R = 1 ,25087   ,51.4,49.9,50.7
XS GIS Cut Line= 4
     2101229.935      182280.066     2101199.987      182793.087
     2101240.351      182811.316     2101198.685      183377.722
#Sta/Elev= 30
       0 2217.07    29.6 2211.71   108.5 2194.45   154.5 2187.52   200.5    2179
   259.6 2161.06   305.6 2151.18   384.7 2138.53   463.4 2128.13     482 2122.34
     510 2121.56   525.6 2121.09  533.742117.908     540 2116.58  545.452117.909
   550.8 2119.87   561.8  2121.1   601.2 2120.81   611.1  2122.2   632.1 2119.32
     713 2119.13   726.2 2121.26   745.9 2122.28   762.4 2128.96   831.7 2166.28
   889.5 2200.43   949.9 2227.53  1058.5 2282.74  1104.5 2305.27  1126.1 2314.66
#Mann= 6 ,-1 , 0
       0      .1       0     510     .04       0  533.74    .045       0
  545.45     .04       0  728.18     .06       0  828.18      .1       0
#XS Ineff= 2 , 0
          519.03  2126.8  560.88         2126.71
Permanent Ineff=
       F       F
Bank Sta=533.74,545.45
XS Rating Curve= 0 ,0
Exp/Cntr=0.5,0.3

Type RM Length L Ch R = 1 ,25037   ,160.5,186,203
XS GIS Cut Line= 4
     2101191.306      182284.406     2101161.358      182819.562
     2101201.723      182837.791      2101162.66      183387.271
#Sta/Elev= 30
       0 2212.41    28.5 2206.94    67.9 2194.68   186.5  2174.4   238.8 2160.03
     270 2153.67     321 2145.89   455.7 2129.56   475.5  2125.3   485.3 2120.82
   501.7 2122.51   514.8    2122   537.4 2119.79  546.582116.148   554.1 2114.97
  561.792116.151   568.5 2120.26   574.6 2120.65   606.6 2121.55   629.6 2119.57
   698.7 2119.27   731.6 2122.14   762.4 2136.61     804 2159.62   830.3 2171.86
   938.8 2228.02   984.9  2248.7  1050.6 2280.98  1100.1 2302.12  1131.2 2313.91
#Mann= 6 ,-1 , 0
       0      .1       0     500     .04       0  546.58    .045       0
  561.79     .04       0  720.28     .06       0  820.28      .1       0
#XS Ineff= 2 , 0
           537.7 2123.73  565.43         2123.88
Permanent Ineff=
       F       F
Bank Sta=546.58,561.79
XS Rating Curve= 0 ,0
Exp/Cntr=0.5,0.3

Type RM Length L Ch R = 1 ,24851   ,335.7,337.6,342.4
XS GIS Cut Line= 4
2101018.45784039182309.1528810492101012.63069826182763.669967235
2101010.68831755182994.8132717492100999.03403329 183400.77084018
#Sta/Elev= 30
       0 2171.74      89 2164.21   108.7 2161.88   138.2 2156.17   171.1 2152.46
   207.2 2149.77   220.3 2147.22   351.7 2136.77   447.7 2127.41   469.6 2126.07
   482.8 2122.69   535.3 2117.63   541.12114.712   545.1 2112.91   548.4 2112.59
   554.9 2112.77   561.5 2114.62   587.8 2114.37   597.6 2115.34   646.3  2116.1
   689.5 2120.93   699.3 2125.89   712.4 2136.79   726.5 2145.89   756.5 2162.82
   784.6 2176.69   814.2 2188.46     870 2205.07  1004.6 2237.89  1091.8  2263.4
#Mann= 6 ,-1 , 0
       0      .1       0     380    .035       0  474.55     .04       0
   541.1    .045       0   561.5     .04       0  574.55      .1       0
#XS Ineff= 2 , 0
                          600.35         2119.61
Permanent Ineff=
       F       F
Bank Sta=541.1,561.5
XS Rating Curve= 0 ,0
Exp/Cntr(USF)=0,0
Exp/Cntr=0.3,0.1

Type RM Length L Ch R = 1 ,24514   ,301.4,296.1,294.9
XS GIS Cut Line= 3
     2100741.031      182309.294     2100690.236      182898.172
      2100641.93      183434.511
#Sta/Elev= 30
       0 2182.44    39.8 2174.39   196.9 2148.25   316.4  2134.5   339.5 2132.89
   378.8 2127.67   402.1 2126.51   421.8 2123.12   444.9 2120.82   454.7 2117.34
   469.3 2117.87   477.8 2116.78   484.4 2117.59   540.4 2111.26   584.6 2110.07
   589.8 2109.18   596.3 2110.12   616.1 2108.37  623.862110.189   672.6 2143.48
   708.3 2164.88   787.4 2207.91   807.2 2217.28     869 2249.44   919.2 2273.82
   961.1 2291.29  1008.1 2307.07  1034.5 2314.45  1087.2 2326.61  1129.6 2338.14
#Mann= 7 ,-1 , 0
       0      .1       0     180    .035       0     280      .1       0
     380     .04       0     480      .1       0   584.6    .045       0
  623.86      .1       0
#XS Ineff= 2 , 0
          545.11 2120.13
Permanent Ineff=
       F       F
Bank Sta=584.6,623.86
XS Rating Curve= 0 ,0
Exp/Cntr=0.3,0.1

Type RM Length L Ch R = 1 ,24218   ,248,247.4,241.3
XS GIS Cut Line= 4
2100319.20078472182373.2514444852100402.72315526182783.093774337
2100470.70648012183016.1794595612100616.38503338183426.021789413
#Sta/Elev= 30
       0 2195.59    34.2 2196.49      69 2194.95     165 2179.62   212.9 2168.56
   237.3 2161.79   292.9 2140.76   303.3 2137.41   313.4 2135.83   353.6 2120.73
   390.4 2116.93   400.4 2114.16   413.8 2114.71     430 2113.93   454.8 2107.32
  469.462106.696   475.3    2106   479.8 2106.63   567.5 2108.25   577.8 2104.68
   584.8 2105.58   619.2 2121.01   736.4 2190.94   826.9 2243.37   915.5 2290.95
   959.2 2311.79   997.5 2327.99  1039.3 2340.74  1067.9 2346.17    1096 2348.88
#Mann= 8 ,-1 , 0
       0      .1       0      20     .12       0     220      .1       0
  418.27     .04       0  469.46    .045       0   479.8     .04       0
  518.27     .06       0  628.27      .1       0
#XS Ineff= 2 , 0
          420.19  2122.8
Permanent Ineff=
       F       F
Bank Sta=469.46,479.8
XS Rating Curve= 0 ,0
Exp/Cntr(USF)=0,0
Exp/Cntr=0.5,0.3

Type RM Length L Ch R = 1 ,23970   ,26.4,26.9,28.3
XS GIS Cut Line= 2
     2099957.102      182531.139     2100603.629      183434.177
#Sta/Elev= 30
       0 2201.09    18.1 2197.25    34.2 2195.73    74.5 2184.47   106.8 2172.03
   190.3 2135.47   227.9 2123.24   292.4 2116.77   300.5 2114.66   324.7 2115.41
   365.1 2110.98   409.4 2108.58  416.59 2105.83   421.6 2103.65  427.58 2105.83
     446 2107.35   518.4 2107.17   538.6 2105.96   550.7 2102.29   574.9 2111.09
   595.1 2121.34   647.9 2153.41   767.9 2221.73   817.6 2248.76   890.1  2285.8
   950.1 2314.11   998.6 2334.46  1042.9 2349.11  1079.3 2355.74  1110.6 2356.92
#Mann= 6 ,-1 , 0
       0      .1       0     190     .04       0     310     .06       0
  416.59    .045       0  427.58     .06       0     550      .1       0
#XS Ineff= 2 , 0
          412.12 2114.59   436.1         2114.65
Permanent Ineff=
       F       F
Bank Sta=416.59,427.58
XS Rating Curve= 0 ,0
Exp/Cntr=0.5,0.3

Type RM Length L Ch R = 1 ,23943   ,191.4,189.3,192.2
XS GIS Cut Line= 2
     2099934.966      182545.461     2100581.494        183448.5
#Sta/Elev= 30
       0 2200.53    20.6  2199.1    42.2 2195.02    77.1 2184.83   117.4 2167.88
   190.6 2131.97   214.3 2124.05   234.5 2120.85   274.8 2118.76   282.9 2115.84
   311.1 2115.95   404.8 2109.22   416.1 2107.73  424.822104.805   432.2 2103.39
     4392104.685   517.2 2105.94   537.1 2101.99     540 2102.08     557 2107.83
   578.3 2118.12   601.7 2131.34     664 2170.26   771.1 2229.32     844 2268.15
   940.4 2316.04   994.5 2339.48  1050.9 2359.57  1075.5 2365.81  1110.6 2369.74
#Mann= 7 ,-1 , 0
       0      .1       0     170     .04       0     290     .06       0
     410      .1       0  424.82    .045       0     439     .06       0
     540      .1       0
#XS Ineff= 2 , 0
          418.24 2110.71     449         2110.76
Permanent Ineff=
       F       F
Bank Sta=424.82,439
XS Rating Curve= 0 ,0
Exp/Cntr=0.5,0.3

Type RM Length L Ch R = 1 ,23754   ,294.9,296.2,283.8
XS GIS Cut Line= 4
2099802.52751581182651.0118860442100014.24701322182987.043748908
2100095.82700305183072.5085001572100474.59124154183525.083205633
#Sta/Elev= 30
       0 2178.67    11.4 2177.63    30.8 2170.88   100.6 2138.97   116.1 2129.47
   131.6 2126.58   143.2  2120.4   189.8 2119.89     212 2117.53   255.7 2120.82
     310 2112.18   433.6  2105.5   440.3  2102.4   453.3  2100.5   467.2 2101.66
   481.1 2100.61   490.4 2102.57   513.6 2102.65   529.6 2100.15   539.2 2103.11
   560.2 2116.12   641.4 2176.48   677.8 2200.41     744 2241.15   803.9 2274.43
   872.4 2308.63   923.2 2329.28   974.3 2345.91  1022.1 2357.73  1105.5 2374.18
#Mann= 5 ,-1 , 0
       0      .1       0     160     .04       0     270      .1       0
   440.3    .045       0   490.4      .1       0
Bank Sta=440.3,490.4
XS Rating Curve= 0 ,0
Exp/Cntr(USF)=0,0
Exp/Cntr=0.3,0.1

Type RM Length L Ch R = 1 ,23458   ,338.8,350,359.2
XS GIS Cut Line= 3
     2099546.328      182808.171     2099906.273      183280.112
     2100311.175      183634.749
#Sta/Elev= 30
       0 2128.13    86.8 2123.94    99.2 2124.46   111.5 2123.36   185.8 2121.03
   234.1 2115.49   288.2 2113.02   312.1 2112.93   391.7 2107.98   412.7 2105.68
   495.3 2104.16     520 2100.69   569.6 2099.36  579.682097.721   585.8 2096.73
     596 2096.72  609.92 2097.72   613.5 2099.34   622.2 2106.68   630.9 2112.59
   723.9  2163.7   757.4 2179.82   792.3 2193.18   843.4  2208.1   870.8 2213.56
   938.1 2229.16  1007.8 2240.88  1040.9 2248.04  1097.6 2264.28  1131.8 2277.04
#Mann= 5 ,-1 , 0
       0      .1       0      80     .04       0      90      .1       0
  579.68    .045       0  609.92      .1       0
Bank Sta=579.68,609.92
XS Rating Curve= 0 ,0
Exp/Cntr=0.3,0.1

Type RM Length L Ch R = 1 ,23108   ,389.2,394.4,392.9
XS GIS Cut Line= 3
     2099467.289      182860.355     2099644.146      183497.263
     2099824.215      183991.166
#Sta/Elev= 30
       0 2126.67     232 2115.25   245.6 2115.69   276.2 2112.86   528.2 2098.19
   589.5 2093.42   623.5 2094.72   637.2 2094.33  643.282092.801   654.2 2091.57
   664.5 2091.62  666.632092.797   671.5 2097.37   685.4 2115.91   695.5 2125.24
   705.7 2136.63   770.8 2190.63   800.7 2212.94   815.7 2225.51   863.5 2259.86
   897.6  2281.1   923.2 2294.83   947.4 2305.69   989.3 2320.49  1048.6 2337.25
  1097.5 2348.33  1118.5 2350.61  1132.4 2349.85  1163.9 2339.15  1186.7 2329.43
#Mann= 3 ,-1 , 0
       0      .1       0  643.28    .045       0  666.63      .1       0
Bank Sta=643.28,666.63
XS Rating Curve= 0 ,0
Exp/Cntr=0.3,0.1

Type RM Length L Ch R = 1 ,22714   ,445.1,458.7,467.8
XS GIS Cut Line= 2
     2099110.877      182911.686     2099421.207      183988.075
#Sta/Elev= 30
       0  2126.8   131.4 2120.31   157.7 2120.58   179.2 2118.91   233.8 2117.08
   240.7 2117.76   329.4 2113.18   390.9 2107.55   438.6  2101.4   520.8 2099.45
     548 2095.09   551.4  2093.2   557.62086.196   561.6 2084.84  576.442086.198
   588.9 2089.35     606 2090.36   653.8 2087.89   660.6 2089.06   682.4 2105.58
   712.3 2126.26   865.5 2227.42   988.4 2304.99    1019 2322.33  1043.4 2333.95
  1060.1 2339.55    1072  2341.5  1080.6 2341.48  1094.3  2337.1  1120.2 2323.65
#Mann= 9 ,-1 , 0
       0      .1       0      70    .035       0     280      .1       0
     380     .12       0     480      .1       0   557.6    .045       0
  576.44      .1       0     990     .12       0    1030      .1       0
#XS Ineff= 2 , 0
                          622.35         2105.63
Permanent Ineff=
       F       F
Bank Sta=557.6,576.44
XS Rating Curve= 0 ,0
Exp/Cntr=0.3,0.1

Type RM Length L Ch R = 1 ,22255   ,562,588.2,555
XS GIS Cut Line= 2
     2099093.516      182922.537     2098785.357      183927.311
#Sta/Elev= 30
       0 2127.11    28.1 2124.35   117.3 2118.26   165.3 2115.89   292.3 2114.01
   378.1 2115.71   498.2 2099.99   553.8  2095.8   604.6  2088.8   693.8 2084.98
   712.8 2083.06     735 2078.74   746.4 2079.71  752.722078.145     759 2076.98
   769.2 2077.01  773.552078.145     783 2084.96   800.2 2102.49   824.3 2124.09
   848.2 2142.67   889.4  2173.4   905.7 2186.95   920.3 2195.67   930.6 2199.46
   937.4 2199.43   951.2  2194.7   982.1 2179.01  1008.1 2162.28    1051 2127.43
#Mann= 7 ,-1 , 0
       0     .06       0      60    .035       0     160      .1       0
     370     .12       0     470      .1       0  752.72    .045       0
  773.55      .1       0
Bank Sta=752.72,773.55
XS Rating Curve= 0 ,0
Exp/Cntr=0.3,0.1

Type RM Length L Ch R = 1 ,21667   ,338.8,317.4,199.9
XS GIS Cut Line= 3
     2099073.985      182911.686     2098624.766      183228.527
     2098509.749      183896.929
#Sta/Elev= 30
       0 2127.54   119.4 2122.34   171.6 2124.09   198.3 2117.94     236 2116.26
   257.2 2110.94     276 2103.06   325.4 2067.87   351.3 2066.82   360.3 2064.95
   392.4 2066.83   428.6 2067.48   448.7 2063.08   497.3 2076.56   572.7 2086.58
   600.1    2093   702.5 2132.03   802.4 2173.15   878.4 2190.18     889 2191.04
   905.6 2187.92   963.7 2166.31  1048.9 2125.56  1065.4 2114.84  1085.4 2094.62
    1092 2090.92  1098.7 2092.06  1128.7  2111.8  1191.9  2127.7  1227.9 2142.91
#Mann= 5 ,-1 , 0
       0     .06       0     100     .04       0     120      .1       0
   351.3    .045       0   392.4      .1       0
Bank Sta=351.3,392.4
XS Rating Curve= 0 ,0
Exp/Cntr=0.3,0.1

Type RM Length L Ch R = 1 ,21349   ,290.2,283.8,276.6
XS GIS Cut Line= 4
2098668.17718105182792.8056778882098551.63433844183053.084693055
2098584.65481051183231.7837183932098435.09149583183880.538875599
#Sta/Elev= 30
       0 2119.94      96 2114.84   110.4  2109.9   142.8  2111.9   164.3  2109.8
   178.7 2102.68   221.9 2101.75   285.2 2080.77   319.8  2063.8  352.84 2058.91
   366.5 2057.99     383 2058.91   409.9 2059.83   449.9 2077.16   581.1 2115.47
   689.9  2161.9     724 2174.03   747.4 2178.24   763.8 2178.89     783 2175.43
   829.5 2158.73   884.2 2131.57   930.7 2103.79   978.4 2081.54   985.1 2082.09
  1012.1 2093.81  1042.9 2118.38  1052.5 2122.96  1106.3  2135.2  1132.7 2130.92
#Mann= 5 ,-1 , 0
       0      .1       0     210     .04       0  315.18      .1       0
  352.84    .045       0     383      .1       0
Bank Sta=352.84,383
XS Rating Curve= 0 ,0
Exp/Cntr(USF)=0,0
Exp/Cntr=0.3,0.1

Type RM Length L Ch R = 1 ,21065   ,227.1,246.7,259.1
XS GIS Cut Line= 4
 2098372.9353131182753.9580636842098308.83674967183224.014195552
2098405.95578517183453.215119356 2098334.0876989183868.884591338
#Sta/Elev= 30
       0  2136.5    77.6 2124.73   200.5 2111.21   313.1 2105.23   362.8  2100.3
   409.1  2092.2   422.4 2085.94   462.1 2084.78   473.5 2078.58   496.8 2061.64
   511.1 2056.53   533.9 2057.17  559.962053.831   568.9 2053.06  580.442053.832
   596.6 2059.24   652.6 2091.46   691.5 2110.92   723.3 2125.08   738.1 2127.05
     778 2119.41   821.3 2103.46   851.3 2090.55   874.6 2072.38   881.2 2070.85
   894.6 2078.72   931.2 2091.66   961.1 2105.19  1044.4 2137.36  1145.2 2183.03
#Mann= 5 ,-1 , 0
       0      .1       0     230     .04       0  534.41      .1       0
  559.96    .045       0  580.44      .1       0
Bank Sta=559.96,580.44
XS Rating Curve= 0 ,0
Exp/Cntr(USF)=0,0
Exp/Cntr=0.3,0.1

Type RM Length L Ch R = 1 ,20819   ,258.3,268.3,268.9
XS GIS Cut Line= 2
     2098353.499      182729.395     2097999.766      183855.697
#Sta/Elev= 30
       0 2141.52      93 2127.36   161.8 2120.17   192.7 2115.44   206.5 2115.62
   251.2 2111.46   302.8 2109.53     375 2104.43   410.6 2100.59   478.2 2087.53
   522.9  2080.9   533.2 2075.15   568.4 2075.78     602 2062.49   615.7 2053.96
     626 2054.41   636.3 2052.45   694.8 2049.01  710.432045.667   725.4 2044.24
  735.892045.667   760.1 2061.48   811.9  2088.8   863.3 2121.64   901.1 2148.56
   911.2 2154.46   934.7 2170.87  1030.8 2228.01  1079.9 2253.76  1180.5 2298.09
#Mann= 6 ,-1 , 0
       0      .1       0     260    .035       0     370     .04       0
     570      .1       0  710.43    .045       0  735.89      .1       0
#XS Ineff= 2 , 0
          695.25 2052.63
Permanent Ineff=
       F       F
Bank Sta=710.43,735.89
XS Rating Curve= 0 ,0
Exp/Cntr=0.3,0.1

Type RM Length L Ch R = 1 ,20550   ,240.4,242.4,241.5
XS GIS Cut Line= 4
2098232.02315664182699.2188088552098039.59098752183092.964631834
2097859.00079803183463.0264955362097731.69951692183750.194501769
#Sta/Elev= 30
       0 2160.92   103.1 2139.99   179.8 2128.17   252.9  2122.5   285.7 2116.11
   322.3 2107.91   366.1 2094.22   428.1 2068.63     440 2062.72   447.3 2057.11
   452.2 2054.98   481.7  2054.7   493.8 2049.22   501.1 2048.19   555.3 2047.06
   563.2 2045.55  571.612040.662   577.3 2039.62   589.32040.661   626.4 2044.62
   639.9 2048.08   654.5 2054.75   672.7 2065.57   712.9  2085.4   789.6 2127.48
     837 2155.84   953.2 2229.51   991.5 2251.83  1095.8 2305.32  1164.1 2338.86
#Mann= 7 ,-1 , 0
       0      .1       0     270     .12       0     310      .1       0
  498.25     .04       0  571.61    .045       0   589.3     .04       0
  638.25      .1       0
Bank Sta=571.61,589.3
XS Rating Curve= 0 ,0
Exp/Cntr(USF)=0,0
Exp/Cntr=0.3,0.1

Type RM Length L Ch R = 1 ,20308   ,356.9,352.7,350.2
XS GIS Cut Line= 3
     2098043.254      182647.938     2097763.197      183115.903
     2097532.524      183621.706
#Sta/Elev= 30
       0 2129.06    72.2 2120.19   106.3 2117.23   144.3 2111.76   228.9 2094.37
   272.1 2082.23   295.3 2074.28   309.7 2067.18   335.9 2049.12   347.5 2049.57
   371.8 2048.38     378 2045.29   407.7 2043.66   504.2 2043.03     531 2039.81
  536.112036.243   540.4 2034.39  557.172036.241   571.5 2044.02   586.6 2055.83
   625.6 2079.98   668.8 2109.19   744.5 2147.85   800.1 2173.58   827.5 2184.88
   925.4 2218.92   950.4 2230.27  1013.6    2262    1051 2279.62  1101.3 2300.98
#Mann= 8 ,-1 , 0
       0     .12       0      60     .04       0     160     .12       0
     250     .04       0     270     .06       0     440      .1       0
  536.11    .045       0  557.17      .1       0
Bank Sta=536.11,557.17
XS Rating Curve= 0 ,0
Exp/Cntr=0.3,0.1
