HEC-RAS study DRPLKCR.prj: DRPLKCR

--- DRPLKCR.g01 (geometry) --- (continued)

Type RM Length L Ch R = 1 ,19955   ,366.6,348.3,331.2
XS GIS Cut Line= 3
     2097639.523      182477.659     2097422.509      183052.745
     2097415.999       183593.11
#Sta/Elev= 30
       0 2209.47    51.8 2216.53    79.7 2218.66    90.4 2217.94   107.9 2213.53
   132.5 2203.12     151 2193.51   192.1 2168.48   276.2 2113.15   349.9 2059.03
   377.9 2040.46   388.4 2035.78   409.5 2036.41   444.6 2034.74   448.8 2034.02
   454.42030.502   476.9 2029.65  482.35  2030.5   518.2 2036.26   525.3 2038.97
     538 2046.38   584.8 2079.16   644.9 2116.22   714.7 2149.32   819.7 2192.31
   891.9 2216.75   950.9 2233.66  1029.7    2252  1088.7 2270.05  1155.1 2283.91
#Mann= 5 ,-1 , 0
       0      .1       0     430     .04       0   454.4    .045       0
  482.35     .04       0     540      .1       0
Bank Sta=454.4,482.35
XS Rating Curve= 0 ,0
Exp/Cntr=0.3,0.1

Type RM Length L Ch R = 1 ,19607   ,351.8,348.4,339.2
XS GIS Cut Line= 3
     2096875.429      182538.409     2097147.731      182992.248
     2097353.927      183599.017
#Sta/Elev= 30
       0  2165.7    16.3 2163.24    35.4 2165.07    87.6 2162.27   156.9 2152.71
   226.3 2139.38   281.3 2122.35   290.9 2118.66   299.4 2113.21   310.9 2111.83
   376.9 2076.11   395.1 2063.11     418 2042.83   429.6 2034.69   439.1 2029.95
     463 2026.48   517.5 2025.43  524.352023.242   539.4 2022.12  544.792023.242
   553.3 2027.45   586.9 2027.93   594.7 2029.65   604.4 2037.12   650.3 2063.15
   716.2 2096.64   809.7 2140.25  1057.6    2247  1104.2 2261.43  1170.1 2275.41
#Mann= 6 ,-1 , 0
       0      .1       0     500     .04       0     520     .06       0
  524.35    .045       0  544.79     .06       0  619.26      .1       0
#XS Ineff= 2 , 0
          476.09 2031.38  567.35         2030.41
Permanent Ineff=
       F       F
Bank Sta=524.35,544.79
XS Rating Curve= 0 ,0
Exp/Cntr=0.3,0.1

Type RM Length L Ch R = 1 ,19259   ,167.4,194,211.3
XS GIS Cut Line= 3
     2096556.267      182814.702      2096921.32      183221.246
     2097268.285      183662.383
#Sta/Elev= 30
       0 2309.24    66.3 2256.91   119.2 2216.92   194.2 2164.92   199.6 2159.47
     213 2154.73   222.3  2147.3   240.9 2134.74   292.9 2102.16   336.2 2072.73
   379.4 2040.61   401.4 2027.74   410.5 2023.61   419.1 2021.58   445.2 2021.17
   467.6  2017.5   524.3 2019.25  539.682016.515   551.1 2015.74   559.92016.514
   567.8  2018.8   588.7 2030.62   651.3 2072.25   688.8 2094.06   781.2 2144.45
   856.2 2182.09   923.7 2209.28   961.1 2220.84  1039.5 2240.67  1107.6 2253.89
#Mann= 6 ,-1 , 0
       0      .1       0     420     .04       0     490     .06       0
  539.68    .045       0   559.9     .06       0  566.39      .1       0
Bank Sta=539.68,559.9
XS Rating Curve= 0 ,0
Exp/Cntr=0.5,0.3

Type RM Length L Ch R = 1 ,19065   ,31.1,33.1,34.4
XS GIS Cut Line= 4
     2096307.192      183057.843     2096810.056      183338.052
     2096792.869      183394.302     2097247.209      183667.705
#Sta/Elev= 30
       0    2317   126.1 2234.05     222 2176.15   238.8 2165.22   247.2 2158.07
   256.9 2155.48   266.5 2148.02   296.1  2129.6   416.1 2061.19   479.1 2021.02
   490.8 2017.87   512.9  2015.1   558.4 2018.22   569.3 2017.85   577.5 2014.29
  582.822014.048   608.3 2011.65   611.8 2011.72  616.282014.054   618.6  2016.7
   622.1 2017.62     671 2017.61   678.7 2019.86   775.3 2084.64   832.7 2119.14
   904.4 2156.13   954.3 2178.35  1018.7  2202.6  1081.3 2222.72  1164.7  2245.7
#Mann= 5 ,-1 , 0
       0      .1       0     500     .06       0  582.82    .045       0
  616.28     .04       0  684.48      .1       0
#XS Ineff= 2 , 0
          573.08  2025.7  623.35         2025.46
Permanent Ineff=
       F       F
Bank Sta=582.82,616.28
XS Rating Curve= 0 ,0
Exp/Cntr=0.5,0.3

Type RM Length L Ch R = 1 ,19032   ,196.8,164.9,136.2
XS GIS Cut Line= 4
     2096298.063      183071.278     2096776.419      183338.052
     2096759.232      183394.302     2097234.478      183680.002
#Sta/Elev= 30
       0  2319.1   140.3  2226.4   194.3  2194.5   234.7 2168.66   241.7 2162.11
   254.9  2157.8   276.1 2142.36   324.4 2112.32   403.3 2068.61   473.1 2023.35
   485.2 2018.27   510.8 2013.92   519.7 2015.79   547.7 2016.45   555.72013.668
   580.4 2012.31  584.962013.669   590.7 2015.32   597.5 2014.59   609.5 2017.72
   678.5 2018.43   693.8 2027.49   751.2 2066.76   804.8 2101.51   850.9 2127.47
   908.2  2155.7   941.6  2170.3  1015.3 2197.37  1072.7 2215.36    1161    2240
#Mann= 6 ,-1 , 0
       0      .1       0     510     .06       0   555.7    .045       0
  584.96     .06       0  587.72     .04       0  696.53      .1       0
#XS Ineff= 2 , 0
          552.86 2020.63  588.45         2020.57
Permanent Ineff=
       F       F
Bank Sta=555.7,584.96
XS Rating Curve= 0 ,0
Exp/Cntr=0.5,0.3

Type RM Length L Ch R = 1 ,18867   ,200.8,192.3,186.7
XS GIS Cut Line= 4
2096245.53107229183214.3449231282096577.10650217183436.382041349
2096876.11648804183593.2882715592097169.20548409 183741.31301704
#Sta/Elev= 30
       0 2273.49    21.2 2257.02    76.5 2217.97    89.8 2207.56   101.6  2203.5
   115.9 2193.27   166.5 2165.45   235.5 2135.33   329.2 2100.46   413.3 2056.53
   448.3 2032.44     474  2017.1   480.6 2014.52   489.1 2013.45  499.632008.576
   515.9 2007.56   524.42008.575   555.8    2011   566.9 2014.38   593.1 2014.31
   600.4 2017.49     615 2026.52   629.5  2040.2   648.4 2053.45     700 2080.94
     752 2104.22   785.1 2116.92   873.2 2147.22  1009.3 2192.36  1065.1 2208.42
#Mann= 7 ,-1 , 0
       0      .1       0  469.05     .04       0  479.05      .1       0
  499.63    .045       0   524.4      .1       0  579.05     .04       0
  699.05      .1       0
Bank Sta=499.63,524.4
XS Rating Curve= 0 ,0
Exp/Cntr(USF)=0,0
Exp/Cntr=0.3,0.1

Type RM Length L Ch R = 1 ,18674   ,225.9,230.6,233
XS GIS Cut Line= 3
     2096076.461      183594.752     2096618.241      183672.383
      2097151.42      183789.178
#Sta/Elev= 30
       0 2357.63      72 2302.78   138.9  2253.9   271.4  2161.1   427.2 2057.22
   462.7 2035.27   487.5 2021.19   503.4 2016.19   513.4 2010.36   523.3 2009.35
   533.6 2004.29   556.6 2003.59  560.692004.291     570 2010.32   580.1 2010.28
     607 2012.35   627.1  2011.7   630.5 2012.79   640.6 2020.98   698.4 2054.21
   731.2 2070.11   771.5 2087.34   838.7 2110.32   909.5 2132.08   979.8 2151.16
   999.9 2155.99  1033.5 2162.56  1046.8 2167.45    1057  2172.2  1093.1 2191.98
#Mann= 5 ,-1 , 0
       0      .1       0   533.6    .045       0  560.69      .1       0
  567.31     .04       0  677.31      .1       0
Bank Sta=533.6,560.69
XS Rating Curve= 0 ,0
Exp/Cntr=0.3,0.1

Type RM Length L Ch R = 1 ,18444   ,241.4,241.6,241.8
XS GIS Cut Line= 4
2096056.05939807183756.1154915882096470.52868542183862.693308334
2096677.76332909183930.7846912552097092.23261644184069.927952007
#Sta/Elev= 30
       0 2348.98    38.3 2319.68   108.8 2270.16   159.6 2236.11     207 2201.77
   251.6 2172.29   301.9 2140.57   366.2 2094.87   399.4 2073.49   420.4 2058.16
   430.7 2054.15     441 2046.86     455  2040.9   489.4 2022.12  528.851998.052
   537.7 1996.87  558.661998.052   575.7 2003.76   603.3 2004.78   617.1 2010.81
   634.6 2011.95   637.9 2013.89   651.7 2026.64   665.5 2036.23   745.1 2082.48
   816.8 2119.84   840.5 2133.44   866.3 2145.96  1025.1 2229.81  1083.3 2257.42
#Mann= 5 ,-1 , 0
       0      .1       0  528.85    .045       0  558.66      .1       0
  607.95     .06       0  716.09      .1       0
Bank Sta=528.85,558.66
XS Rating Curve= 0 ,0
Exp/Cntr(USF)=0,0
Exp/Cntr=0.3,0.1

Type RM Length L Ch R = 1 ,18202   ,80.7,80.6,80.8
XS GIS Cut Line= 3
     2096006.834      183962.629     2096527.388      184134.278
     2097037.796      184326.382
#Sta/Elev= 30
       0 2278.92    83.3 2225.78   114.4 2213.66     149 2202.36   211.2 2168.55
   252.4 2142.54   307.3 2105.19   386.4 2058.09   446.1 2020.42   463.1 2007.26
   480.6 2000.49   508.2 1999.49   522.1 1996.27  531.861995.416   542.8 1994.55
  556.781995.415   591.8 2001.89   630.3 2002.52   640.6 2006.28   661.9 2007.81
     666 2010.28   675.9 2019.86   686.4 2026.33     718 2043.26   812.6  2098.3
   840.7 2111.78   881.9 2133.62   928.4 2160.77  1076.1 2255.55  1093.5 2267.71
#Mann= 6 ,-1 , 0
       0      .1       0  531.86    .045       0  556.78      .1       0
  618.12     .04       0  668.12     .06       0  778.12      .1       0
#XS Ineff= 2 , 0
          498.57 2025.72
Permanent Ineff=
       F       F
Bank Sta=531.86,556.78
XS Rating Curve= 0 ,0
Exp/Cntr=0.5,0.3

Type RM Length L Ch R = 1 ,18122   ,15.4,15.5,16.1
XS GIS Cut Line= 4
2095992.25041816184005.2429211532096458.11295008184194.986323209
2096588.38453955184241.7141759552097003.27123211184393.225698492
#Sta/Elev= 30
       0 2260.64      41 2235.35   101.2 2190.04   122.4 2176.29   203.2 2144.55
   236.3 2127.85   305.9 2085.31   359.8 2047.95   395.2 2028.65   410.2 2016.97
   417.2 2012.91   444.8 2001.45   520.6 1996.46   532.9 1993.66   553.8 1993.52
   564.5 1996.31   569.5 1999.31   578.2 2001.08   616.5 2001.19     627 2002.32
   637.5 2006.07   656.7 2007.79   661.8 2011.63   669.4 2020.27   675.9  2025.2
   689.7 2031.47   794.6 2088.85     868 2125.75   983.2 2188.51  1083.1 2253.54
#Mann= 7 ,-1 , 0
       0      .1       0     410     .06       0   520.6    .045       0
   564.5     .06       0  593.02     .04       0  691.42     .06       0
  701.42      .1       0
#XS Ineff= 3 ,-1
  445.39   491.5 2000.96  497.62  518.111996.481  566.49   585.71996.065
Permanent Ineff=
       F       F       F
Bank Sta=520.6,564.5
XS Rating Curve= 0 ,0
Exp/Cntr(USF)=0,0
Exp/Cntr=0.5,0.3

Type RM Length L Ch R = 1 ,18106   ,27.6,28.9,30.7
XS GIS Cut Line= 4
 2095993.6664137184017.9868809922096453.86496347184209.146278587
2096584.13655294184258.7061224072096989.11127673184421.545609247
#Sta/Elev= 30
       0 2249.57    14.7 2242.92    23.6 2236.42    33.7 2230.94   121.3 2167.11
   139.2  2158.8   195.9    2137   249.2 2110.85   309.6 2074.16     336 2056.24
   355.7 2040.92   394.8  2018.3   412.7 2006.56   438.6 2000.19   487.2 1999.32
   510.7  1996.1   525.9 1993.99   544.6 1993.76     554  1994.3   558.9 1996.17
   571.6 2000.65   620.7 2001.93   631.2 2005.77   650.5 2007.51   666.5 2021.65
   680.7 2030.18   783.2 2085.55   917.8 2156.05  1013.7 2209.39  1074.2 2247.27
#Mann= 7 ,-1 , 0
       0      .1       0     380     .06       0   510.7    .045       0
   558.9     .06       0  598.32     .04       0   637.7     .06       0
   697.7      .1       0
#XS Ineff= 3 ,-1
  437.57  486.39  2000.2  492.22  509.191996.103  559.75  593.691996.192
Permanent Ineff=
       F       F       F
Bank Sta=510.7,558.9
XS Rating Curve= 0 ,0
Exp/Cntr(USF)=0,0
Exp/Cntr=0.5,0.3

Type RM Length L Ch R = 1 ,18077   ,13.9,13.2,12.7
XS GIS Cut Line= 4
2095988.00243155184023.6508631432096445.36899024184234.634198266
2096569.97659756184289.8580242382096972.11933028184444.201537851
#Sta/Elev= 30
       0 2247.86    15.9 2239.74    57.3 2211.85    82.6 2192.95   100.7 2181.69
   122.3 2164.01   133.2 2156.79   211.2 2123.25     255 2101.64   331.9 2056.05
   357.1 2039.14   382.5 2019.75   406.5 2006.87   422.2  2001.8   436.7 1999.96
   483.6 1999.59   512.9 1994.86  525.861994.225   544.8 1993.52  558.451994.225
   577.5 1999.32   619.8 2000.13   632.2 2004.74   655.7 2007.12   676.8  2022.9
   711.9 2043.79   828.5 2107.01   929.8  2159.6  1028.2 2214.13  1070.7 2239.21
#Mann= 7 ,-1 , 0
       0      .1       0     400     .06       0  525.86    .045       0
  558.45     .06       0  563.68     .04       0  613.68     .06       0
  719.98      .1       0
#XS Ineff= 2 , 0
          511.97 1994.34  571.02         1994.48
Permanent Ineff=
       F       F
Bank Sta=525.86,558.45
XS Rating Curve= 0 ,0
Exp/Cntr(USF)=0,0
Exp/Cntr=0.5,0.3

Type RM Length L Ch R = 1 ,18064   ,23.9,25.2,29.5
XS GIS Cut Line= 4
 2095982.3384494184029.3148452942096429.79303932184243.130171492
2096581.30456186 184306.849970692096966.45534813184459.777488766
#Sta/Elev= 30
       0 2244.91    31.2 2228.12   100.3 2181.57   122.1 2164.25   144.5 2149.03
   173.7 2134.27   227.4 2111.69   264.3 2093.23   303.1 2071.71   352.9 2041.51
   387.3 2015.83   402.2    2007   429.1 1999.94   488.2 1999.32  525.15 1993.33
   535.3 1992.42  561.061993.331   571.4 1997.06   582.1 1999.25   621.2 2000.13
   635.4 2004.73   658.4 2006.96     671 2017.02   752.1 2063.72   882.7 2133.02
   932.2 2158.05  1012.1 2202.79    1031 2212.35  1048.7 2223.65  1074.7 2237.28
#Mann= 6 ,-1 , 0
       0      .1       0     400     .06       0  525.15    .045       0
  561.06     .04       0  615.92     .06       0  730.28      .1       0
#XS Ineff= 2 , 0
          519.78 1993.39  564.67         1993.61
Permanent Ineff=
       F       F
Bank Sta=525.15,561.06
XS Rating Curve= 0 ,0
Exp/Cntr(USF)=0,0
Exp/Cntr=0.5,0.3

Type RM Length L Ch R = 1 ,18039   ,25.1,27.5,27.3
XS GIS Cut Line= 4
2095980.44840669184034.8129627922096441.12100363184271.450082247
2096595.46451724184364.9057877382096914.06351323184536.241247804
#Sta/Elev= 30
       0 2240.86    15.4 2234.04    30.1 2225.52   100.7 2178.11   120.2 2162.86
   159.2 2136.93     185 2123.79   251.4 2094.32   295.7 2069.85   345.8 2040.34
   395.5 2005.01   424.8 1999.25   490.5 1998.95   517.9 1995.27   535.31992.973
   539.9 1992.06  560.281992.973   586.6 1997.93   617.7 1999.99   629.6 2003.75
   651.2 2005.47   670.2 2017.93   693.4 2028.72   738.2 2053.45   873.3 2124.03
   916.9  2143.9   943.1 2152.98   973.7 2166.84    1025 2191.79  1060.1 2210.71
#Mann= 7 ,-1 , 0
       0      .1       0     410     .06       0   517.9     .04       0
   535.3    .045       0  560.28     .04       0   637.9     .06       0
   687.9      .1       0
#XS Ineff= 2 , 0
          518.18 1995.23  577.93         1996.13
Permanent Ineff=
       F       F
Bank Sta=535.3,560.28
XS Rating Curve= 0 ,0
Exp/Cntr(USF)=0,0
Exp/Cntr=0.5,0.3

Type RM Length L Ch R = 1 ,18011   ,109.4,114.2,116.6
XS GIS Cut Line= 4
2095975.25847171184039.2268140592096431.20903486184292.690015313
2096545.90467342184367.7377788132096891.40758463184578.721113936
#Sta/Elev= 30
       0 2238.01    25.7 2226.36    54.4 2208.15   102.7 2175.74   167.8 2129.63
     216 2104.92   261.8 2083.59   295.7 2065.53   340.6 2038.25   384.9 2005.64
   390.3 2003.67   421.1 1999.03   490.8 1998.02  542.841992.616     556 1991.55
  570.581992.615   583.5 1997.62   614.9 1998.78   629.1 2003.59   652.8 2005.75
     663 2013.33   681.9  2020.8   715.7 2040.41   791.2 2077.36   842.5    2106
     877 2123.01     904 2135.35   958.9 2155.56  1008.4 2176.75  1063.6 2204.36
#Mann= 6 ,-1 , 0
       0      .1       0     430     .06       0  541.67     .04       0
  542.84    .045       0  570.58     .04       0  651.67      .1       0
#XS Ineff= 2 , 0
          532.11 1993.73  577.54         1993.87
Permanent Ineff=
       F       F
Bank Sta=542.84,570.58
XS Rating Curve= 0 ,0
Exp/Cntr(USF)=0,0
Exp/Cntr=0.5,0.3

Type RM Length L Ch R = 1 ,17897   ,148.8,147.5,145.9
XS GIS Cut Line= 3
     2095963.078      184049.555     2096396.146       184395.61
     2096751.716      184808.891
#Sta/Elev= 30
       0 2231.94    11.9 2225.82    22.9 2222.01    66.5 2195.88    93.6 2175.88
   145.4 2140.47     173 2119.37   203.4 2100.37     236 2077.37   304.3 2046.77
   318.8 2037.36   336.4 2021.37   345.7 2014.75   358.9 2011.79   369.1 2004.44
   397.6 1997.59   505.9 1995.39  563.571990.613   572.1 1989.28  579.061990.614
   591.9  1998.5   604.7 2000.14     614 2004.01     633 2004.25   651.2 2013.86
   702.5 2030.34   775.9 2048.39   873.6 2075.61   972.3 2112.38  1099.5  2164.5
#Mann= 5 ,-1 , 0
       0      .1       0     490     .04       0  563.57    .045       0
  579.06     .04       0  634.35      .1       0
#XS Ineff= 2 , 0
          502.87  1998.3
Permanent Ineff=
       F       F
Bank Sta=563.57,579.06
XS Rating Curve= 0 ,0
Exp/Cntr=0.3,0.1

Type RM Length L Ch R = 1 ,17750   ,101.9,106,111.6
XS GIS Cut Line= 4
2095912.95466805184115.6905730962096264.12156141184473.937444143
2096400.05713303 184607.04102469 2096646.4403566 184907.23207869
#Sta/Elev= 30
       0  2204.5     8.1 2197.53      62 2161.36    95.7  2143.3   104.9 2136.82
   117.2 2133.16   181.5 2093.23   213.6 2076.62   288.2 2043.28   300.9    2038
   317.5 2034.84   364.8 2009.99   397.1 1999.04   411.2 1995.89     439 1993.17
   498.5 1993.79   534.1 1991.32  543.381987.209   552.7 1986.22  560.611987.208
   573.6 1988.96   592.1  1996.8   619.7 1997.57   628.8 2002.82   645.5  2008.1
     714 2026.11   745.5 2040.44   796.7    2060   877.5 2094.71  1080.3 2169.47
#Mann= 6 ,-1 , 0
       0      .1       0     480     .06       0  543.38    .045       0
  560.61     .06       0  611.66     .04       0  621.66      .1       0
#XS Ineff= 2 , 0
          486.53 2006.95
Permanent Ineff=
       F       F
Bank Sta=543.38,560.61
XS Rating Curve= 0 ,0
Exp/Cntr(USF)=0,0
Exp/Cntr=0.5,0.3

Type RM Length L Ch R = 1 ,17644   ,38.5,37.3,36.1
XS GIS Cut Line= 4
2095836.49090901 184200.650305362096203.23375329184550.401203181
2096281.11350786184655.1848729732096565.72861095 184995.02380203
#Sta/Elev= 30
       0 2170.16    31.9 2152.27   126.5 2120.06   149.8 2109.87     157 2107.89
   188.3 2093.59   245.2  2070.3   258.6 2062.17   282.3 2054.99     389 2006.63
   414.6 1996.05   480.7 1990.98   535.7 1988.82   543.6 1986.83   551.9 1984.83
     566 1984.57   570.7 1984.93  574.59 1986.88   582.4 1990.07   608.2 1990.28
   625.3 1993.32   676.1 2019.82   721.7 2041.32   778.4 2066.95   790.1 2070.59
   808.6 2079.66   854.6 2098.95   964.7 2142.01  1007.9 2157.25  1080.6 2180.34
#Mann= 5 ,-1 , 0
       0      .1       0   543.6    .045       0  574.59      .1       0
  576.78     .04       0  636.78      .1       0
#XS Ineff= 2 , 0
          527.67 1987.45  584.55         1987.45
Permanent Ineff=
       F       F
Bank Sta=543.6,574.59
XS Rating Curve= 0 ,0
Exp/Cntr(USF)=0,0
Exp/Cntr=0.5,0.3

Type RM Length L Ch R = 1 ,17606   ,102.9,104,105.4
XS GIS Cut Line= 4
2095830.82692686184220.4742428892096170.66585592184573.057131785
 2096271.2015391184696.2487435682096527.49673143185023.343712785
#Sta/Elev= 30
       0 2162.41    34.5 2148.25    84.6 2131.41   142.3 2109.43   151.6 2106.87
   221.3  2077.7   244.7  2065.9   262.3  2061.7   339.5 2026.13     372 2009.95
     399 1998.83   418.4 1994.62     481  1990.1     516 1989.45   532.5 1985.76
   542.5 1983.88   556.8 1984.16   562.1 1985.66   569.6 1988.64   594.4  1989.1
   616.3 1996.21   630.3 2002.81   651.2 2015.92   688.6 2035.91   777.4 2078.18
   788.5 2081.08   813.5 2092.75   910.6 2130.12  1021.9 2168.72  1064.3 2180.95
#Mann= 5 ,-1 , 0
       0      .1       0   532.5    .045       0   562.1      .1       0
   589.7     .04       0   609.7      .1       0
#XS Ineff= 2 , 0
          527.92 1986.03  564.83         1986.11
Permanent Ineff=
       F       F
Bank Sta=532.5,562.1
XS Rating Curve= 0 ,0
Exp/Cntr(USF)=0,0
Exp/Cntr=0.5,0.3

Type RM Length L Ch R = 1 ,17502   ,186.4,184.9,183.5
XS GIS Cut Line= 3
     2095800.892      184241.614     2096124.973      184681.383
     2096446.087      185122.912
#Sta/Elev= 30
       0 2165.81   175.7 2105.45   222.9 2082.74     237 2074.28   251.1 2071.77
   269.5 2062.72   292.5 2053.94   306.1 2046.52   330.6 2036.56   346.9 2031.93
   436.4 1992.78   447.3 1990.72   520.9  1987.8  534.781982.113   546.6 1980.96
  554.281982.113   562.8  1985.4   583.1 1985.18   591.2 1987.82     636 2015.55
     664 2035.81   687.6 2050.45   729.9 2072.07   814.6 2106.26   831.4 2110.19
   866.1 2122.86   932.5 2143.98  1013.1 2166.76  1051.5 2174.63  1092.2 2180.58
#Mann= 5 ,-1 , 0
       0      .1       0     510     .04       0  534.78    .045       0
  554.28     .04       0  756.28      .1       0
Bank Sta=534.78,554.28
XS Rating Curve= 0 ,0
Exp/Cntr=0.3,0.1

Type RM Length L Ch R = 1 ,17317   ,169.3,165.1,160.6
XS GIS Cut Line= 4
2095628.91767081184407.4198906672095948.30333099184758.272118351
2096094.62286989184929.7649112542096360.51536531185198.804063424
#Sta/Elev= 30
       0 2157.18    29.2  2149.4    50.8 2141.71    64.7 2138.92   101.9 2126.02
   113.6 2123.98   126.8 2118.24   187.9  2099.3   266.8 2070.24   366.7  2037.7
   401.9 2024.03   446.2 2001.03   474.5 1990.38   489.8 1985.51  516.851979.892
   524.7 1978.89  538.611979.892   550.3 1982.81   570.3 1982.95   589.4 1988.52
   606.6 2001.04   632.5 2016.08   685.3 2039.67   748.2  2071.8     799 2094.23
   868.6 2118.89   906.9 2129.25   946.1 2137.05  1033.7  2142.6  1078.1 2142.56
#Mann= 5 ,-1 , 0
       0      .1       0  516.85    .045       0  538.61      .1       0
  594.45     .04       0  729.88      .1       0
Bank Sta=516.85,538.61
XS Rating Curve= 0 ,0
Exp/Cntr(USF)=0,0
Exp/Cntr=0.3,0.1

Type RM Length L Ch R = 1 ,17152   ,362.3,350,341.9
XS GIS Cut Line= 3
     2095434.697      184580.102     2095865.522      184913.644
     2096307.943      185244.622
#Sta/Elev= 30
       0 2234.97   101.6 2196.07   118.3 2186.42   134.4 2180.78   172.2 2162.25
   181.1 2159.84     193 2152.47   260.7 2118.11   342.7 2070.57   450.1 2024.87
   473.5  2009.4   494.5 1992.17   508.3 1982.59   516.6 1979.44  532.671977.106
   545.6 1976.22  553.621977.105   574.3  1981.3   639.9  1980.1   660.4 1981.94
   680.8 1998.62   705.3 2014.03   776.4 2050.29   834.3 2074.26   877.5 2089.65
   902.2 2096.77   930.8 2101.78   963.2 2104.77  1028.4 2107.55  1097.4    2107
#Mann= 6 ,-1 , 0
       0      .1       0     530     .04       0  532.67    .045       0
  553.62     .04       0  604.85     .06       0  654.85      .1       0
#XS Ineff= 2 , 0
                          584.53         1993.05
Permanent Ineff=
       F       F
Bank Sta=532.67,553.62
XS Rating Curve= 0 ,0
Exp/Cntr=0.3,0.1

Type RM Length L Ch R = 1 ,16802   ,340.4,350,353.1
XS GIS Cut Line= 3
     2095186.036      185165.385     2095727.595      185229.638
     2096266.273      185338.859
#Sta/Elev= 30
       0 2203.63      77 2186.24   119.9 2173.75   133.1 2167.84   199.2  2144.6
   242.2 2126.91   268.3 2113.19   285.1 2106.63   341.3 2076.61   384.2 2050.57
   410.7 2035.87   456.9 2005.85   492.8 1980.86   509.8 1973.85  531.491971.601
   539.5 1970.19  552.831971.603   559.5 1974.24   579.6 1974.95     635 1974.06
   649.9 1981.23   663.3 1983.48   696.8 1992.02   726.9 1995.01   792.5 2010.96
   840.7 2017.79   867.5 2024.46   897.6  2035.4   974.8 2048.44    1095 2077.19
#Mann= 6 ,-1 , 0
       0      .1       0  531.49    .045       0  552.83      .1       0
  575.36     .06       0  605.36     .04       0  675.36      .1       0
#XS Ineff= 2 , 0
                          581.09         1988.41
Permanent Ineff=
       F       F
Bank Sta=531.49,552.83
XS Rating Curve= 0 ,0
Exp/Cntr=0.3,0.1

Type RM Length L Ch R = 1 ,16452   ,518.7,519.3,522.1
XS GIS Cut Line= 3
     2095156.447      185279.904     2095648.835      185563.052
     2096154.589      185758.258
#Sta/Elev= 30
       0 2188.84      39 2179.13    73.1 2168.45   175.3 2135.63   201.8 2125.23
   224.5 2114.32   247.4 2099.36   353.1 2039.33   412.3 2002.39   432.6 1987.41
   466.1 1971.12   478.1 1969.17   515.9 1969.28  557.051967.151   563.7 1966.05
  580.74 1967.15   589.8 1970.37     611 1970.29   614.5 1971.57   622.8 1978.48
   642.7 1992.09   688.4    2015   721.7 2026.81   780.7 2043.64   793.9 2046.64
   804.5 2047.43   850.2 2058.59  1001.4 2088.27  1059.9 2101.13  1110.1 2108.22
#Mann= 6 ,-1 , 0
       0      .1       0  557.05    .045       0  580.74     .04       0
     688      .1       0     768     .12       0     998      .1       0
#XS Ineff= 2 , 0
                          598.14         1972.47
Permanent Ineff=
       F       F
Bank Sta=557.05,580.74
XS Rating Curve= 0 ,0
Exp/Cntr=0.3,0.1

Type RM Length L Ch R = 1 ,15933   ,157.9,164.9,171.9
XS GIS Cut Line= 3
     2095119.992      185420.367     2095265.391       185932.52
     2095896.902      186290.593
#Sta/Elev= 30
       0 2173.44    50.6  2164.4   142.7 2141.64     245  2122.2   316.6 2106.41
   360.9 2094.65   381.4 2086.59   391.2  2085.2   476.9 2047.66   540.4 2024.74
   563.9 2014.24   616.3 1985.61   647.5  1963.6  661.991958.359   668.6 1957.23
  681.621958.358   688.5 1959.85   740.2 1960.11   758.3 1963.08     778 1962.64
     793 1967.09   902.4 2029.29   962.8 2057.72   996.5 2077.37  1037.4 2095.67
  1068.7 2107.12  1128.9 2123.69  1158.9 2129.47  1201.1 2133.81  1258.4 2133.52
#Mann= 5 ,-1 , 0
       0      .1       0  661.99    .045       0  681.62      .1       0
  732.39     .06       0  932.39      .1       0
#XS Ineff= 2 , 0
                          754.15         1974.83
Permanent Ineff=
       F       F
Bank Sta=661.99,681.62
XS Rating Curve= 0 ,0
Exp/Cntr=0.3,0.1

Type RM Length L Ch R = 1 ,15768   ,221.9,236.1,248.5
XS GIS Cut Line= 4
2095111.48198097185434.6835281132095193.04332394186019.631284752
2095398.22107736186264.3153136722095640.35631431186523.017698417
#Sta/Elev= 30
       0 2172.68    74.4  2155.2    87.7 2149.55   134.1 2140.13   243.4 2125.48
   293.1 2117.11   319.6 2110.17   369.3 2094.32   418.9 2073.81   455.4 2060.55
   471.9 2056.78     506 2043.41   581.3 2022.39   627.2 2006.68   659.9 1993.87
   696.2 1973.87   715.5 1960.52  727.65 1955.03   735.8 1954.02  746.711955.031
   762.6 1958.69   852.2 1957.93   868.5 1962.34   889.5 1962.91   897.8 1967.64
     929  1976.5     971  1998.4  1159.8 2083.24  1205.8 2097.83  1264.3 2109.52
#Mann= 5 ,-1 , 0
       0      .1       0  727.65    .045       0  746.71      .1       0
  850.61     .06       0  999.93      .1       0
#XS Ineff= 2 , 0
                          818.34         1973.18
Permanent Ineff=
       F       F
Bank Sta=727.65,746.71
XS Rating Curve= 0 ,0
Exp/Cntr(USF)=0,0
Exp/Cntr=0.3,0.1

Type RM Length L Ch R = 1 ,15532   ,285.8,298.1,307.4
XS GIS Cut Line= 2
     2095100.461      185431.218     2095104.801      186776.704
#Sta/Elev= 30
       0 2174.11    77.2 2151.61   162.5 2131.01   201.9 2126.33   251.1 2124.23
     300  2115.6   369.3 2091.23     402 2076.28     435 2068.26   555.7 2029.24
     589 2015.83   684.1    1984   739.9 1974.85   756.3 1967.64   772.7 1954.66
  823.551951.265   831.8 1949.94     8421951.267   848.2 1953.71   864.6  1954.6
     876 1952.41   897.4 1955.93  1041.8 1954.57  1156.6 1961.82  1182.8  1971.4
  1222.2 1974.78  1251.2 1984.91  1274.7  1984.6  1314.1 1999.92  1345.5 2006.81
#Mann= 7 ,-1 , 0
       0      .1       0  823.55    .045       0     842      .1       0
     900    .035       0    1090     .04       0    1190    .035       0
    1290      .1       0
#XS Ineff= 2 , 0
                          896.17         1959.87
Permanent Ineff=
       F       F
Bank Sta=823.55,842
XS Rating Curve= 0 ,0
Exp/Cntr=0.3,0.1

Type RM Length L Ch R = 1 ,15234   ,212.6,213.3,213.1
XS GIS Cut Line= 4
2095093.35723809185446.4362910762094938.16412715186027.277660655
2094852.77959622186158.5404470032094631.03469502 186543.40803416
#Sta/Elev= 30
       0 2170.74    81.1 2144.18   155.8 2123.48     183 2120.81   236.7 2119.29
   264.5 2115.03   325.6 2088.22     352  2079.3   468.3 2027.35   488.7 2020.67
   502.1  2018.5   512.8 2014.16   566.7 1988.11   620.2 1964.52  650.51 1946.52
   659.3 1945.45  670.751946.521   690.6  1949.1   726.9 1950.53   757.2 1948.61
   836.7 1949.02   957.9 1946.86   999.5 1948.74  1031.6 1952.77  1048.8 1956.41
  1074.8 1968.68  1084.4 1971.42  1166.1  2012.3  1187.7 2027.08    1202 2028.86
#Mann= 6 ,-1 , 0
       0      .1       0  650.51    .045       0  670.75      .1       0
  721.22    .035       0 1127.81      .1       0 1177.81     .06       0
#XS Ineff= 2 , 0
                          914.61         1968.87
Permanent Ineff=
       F       F
Bank Sta=650.51,670.75
XS Rating Curve= 0 ,0
Exp/Cntr(USF)=0,0
Exp/Cntr=0.3,0.1

Type RM Length L Ch R = 1 ,15021   ,326.6,318.3,308.4
XS GIS Cut Line= 2
       2095083.1      185444.239     2094421.207      186414.291
#Sta/Elev= 30
       0 2170.83    46.9 2155.43   125.3 2134.23     165 2126.94   231.1 2120.75
   257.1 2112.33   304.3 2090.63   339.8 2071.61   360.9 2064.62     421 2031.08
   443.6 2020.57   476.6 2001.91   546.4 1966.87   566.5 1953.02   582.1 1944.34
     597 1942.68   613.1 1944.43   627.7 1947.77     733 1944.21   796.6 1945.16
   939.4 1944.34   971.3 1945.75   983.3 1942.89  1011.1 1948.97  1032.2 1947.66
  1042.8 1948.85  1067.1 1957.95  1084.6 1960.59  1125.3 1976.54  1174.4 1991.04
#Mann= 5 ,-1 , 0
       0      .1       0   582.1    .045       0   613.1      .1       0
     710    .035       0     950      .1       0
#XS Ineff= 2 , 0
                          627.59         1950.28
Permanent Ineff=
       F       F
Bank Sta=582.1,613.1
XS Rating Curve= 0 ,0
Exp/Cntr=0.3,0.1

Type RM Length L Ch R = 1 ,14702   ,343.9,350,347.5
XS GIS Cut Line= 3
     2094575.726      185295.593     2094451.872      185826.773
     2094328.768      186360.113
#Sta/Elev= 30
       0 2169.52    42.5  2154.4    73.7 2138.91   135.3 2103.17   157.9 2093.78
   194.9  2075.6   252.2 2052.16   282.5 2031.78   334.8 2002.11   356.6 1987.83
   417.3 1959.13   437.5 1950.47   447.6 1948.76   464.4 1942.96  532.291940.054
   548.7 1938.38  556.86 1940.06   565.5 1941.57   592.4 1939.91   631.9 1941.03
   686.7 1939.07   737.2 1941.57   860.8 1940.39   892.6 1943.15     909 1948.86
   929.2 1961.99   952.8 1979.95   996.5 2002.92  1053.7 2029.24  1092.8 2042.04
#Mann= 8 ,-1 , 0
       0      .1       0  532.29    .045       0  556.86    .035       0
  655.43      .1       0  755.43    .035       0  855.43      .1       0
  955.43     .08       0 1055.43      .1       0
#XS Ineff= 2 , 0
                          567.71         1944.41
Permanent Ineff=
       F       F
Bank Sta=532.29,556.86
XS Rating Curve= 0 ,0
Exp/Cntr=0.3,0.1

Type RM Length L Ch R = 1 ,14352   ,197.8,203.6,212.3
XS GIS Cut Line= 3
     2094332.604      185251.212     2094105.668      185793.821
     2094028.303      186326.796
#Sta/Elev= 30
       0  2107.8   111.6 2069.73     165 2045.93   207.7 2024.23     243 2001.91
   268.2 1982.87   302.5 1960.35   318.4 1952.44   332.1 1943.24   339.2  1941.8
   349.9 1936.97     361 1935.68   549.1  1936.7   577.5 1934.06   591.5 1932.59
   603.8 1933.88   608.1 1934.42   624.1  1931.8   631.3 1933.51   644.5 1941.25
   661.7  1948.3   690.9 1955.15   780.5 1961.35     860    1975     923 2000.91
   974.4 2020.32  1024.8 2044.65  1088.8 2072.45  1106.3 2077.47  1126.7 2085.67
#Mann= 5 ,-1 , 0
       0      .1       0   577.5    .045       0   603.8      .1       0
  828.15     .08       0 1028.15      .1       0
#XS Ineff= 2 , 0
          491.69 1952.43
Permanent Ineff=
       F       F
Bank Sta=577.5,603.8
XS Rating Curve= 0 ,0
Exp/Cntr=0.3,0.1

Type RM Length L Ch R = 1 ,14149   ,299.3,292.1,285.4
XS GIS Cut Line= 2
     2094197.683      185179.482       2093687.7      186171.235
#Sta/Elev= 30
       0 2047.17    30.5 2040.34    52.6 2037.29    91.9 2028.41   200.2 1998.38
   279.5 1971.95   296.5 1962.97   323.3 1943.44     344 1937.85   373.6 1935.39
   454.9 1932.32   535.9 1932.71   569.1 1931.74  579.471930.298   591.2 1929.15
  602.811930.297   609.7  1933.2   631.8 1935.51   666.8 1947.19   704.8 1957.36
   799.6 1975.78   845.8 1990.42   888.6 2005.44   926.9 2019.28     986 2042.61
  1007.9 2048.39  1030.2 2049.65  1041.3 2047.45  1066.4 2039.22  1115.2 2011.54
#Mann= 3 ,-1 , 0
       0      .1       0  579.47    .045       0  602.81      .1       0
Bank Sta=579.47,602.81
XS Rating Curve= 0 ,0
Exp/Cntr=0.3,0.1

Type RM Length L Ch R = 1 ,13856   ,240.6,237.8,228
XS GIS Cut Line= 4
2093848.88421168 185006.75128634  2093784.138188185373.645420489
2093724.18816608185882.0216063692093683.42215118  186157.7917072
#Sta/Elev= 30
       0 2110.83    45.4 2093.53      93 2077.93   176.3 2046.49   209.6 2033.36
   269.5 2007.16   336.2 1986.74   369.5 1974.18     386 1966.32   399.2 1961.85
   415.8  1953.5   435.6 1941.83   452.1 1928.58  457.631926.028   468.5 1924.81
  481.671926.028   527.6 1929.32   713.1  1931.3   789.1  1936.3   811.3 1942.39
   841.9 1948.29   871.7 1958.08   934.6 1984.56  1010.9 2020.57    1044 2034.72
  1087.4  2048.6  1100.4 2048.93  1123.7 2042.85  1143.6  2032.8  1163.2 2020.37
#Mann= 5 ,-1 , 0
       0      .1       0  457.63    .045       0  481.67      .1       0
  542.56    .035       0  642.56      .1       0
#XS Ineff= 2 , 0
                          630.95          1958.5
Permanent Ineff=
       F       F
Bank Sta=457.63,481.67
XS Rating Curve= 0 ,0
Exp/Cntr(USF)=0,0
Exp/Cntr=0.3,0.1

Type RM Length L Ch R = 1 ,13619   ,363.7,371.6,379.7
XS GIS Cut Line= 2
     2093464.176      184945.107      2093679.02      186186.426
#Sta/Elev= 30
       0 2038.04   101.7 2021.24   152.1 2009.99   255.4 1989.75   275.3 1984.28
   300.3 1979.75   312.3 1975.64   338.6 1970.87   388.3 1958.69   478.4  1943.7
   495.1 1937.56  521.421922.863   535.1 1921.67  549.091922.862     565 1925.66
   584.2 1926.64   801.4 1928.01     878 1930.06   891.3 1931.89     918 1939.68
   961.7 1957.08   997.9 1974.35  1057.2 2006.79  1107.7 2031.72    1141  2045.1
    1161 2049.68  1174.6 2049.29  1194.3 2042.79    1221 2028.13  1259.8 2002.99
#Mann= 7 ,-1 , 0
       0      .1       0     300    .035       0     500      .1       0
  521.42    .045       0  549.09      .1       0     600    .035       0
     900      .1       0
#XS Ineff= 2 , 0
                           745.6         1930.33
Permanent Ineff=
       F       F
Bank Sta=521.42,549.09
XS Rating Curve= 0 ,0
Exp/Cntr=0.3,0.1

Type RM Length L Ch R = 1 ,13247   ,300.9,295.9,287.1
XS GIS Cut Line= 3
     2093288.395      184940.7662093169.74231116 185619.01777017
2093329.29894279186066.145866133
#Sta/Elev= 30
       0  2029.5  50.0192006.541 132.0831975.682 166.5921961.345 173.2541959.893
 193.2381951.984 216.5521949.089 236.5361948.631 283.1651950.787 319.8031951.198
 363.101 1949.62 393.0771947.056 403.0691942.568 419.7221928.689 429.7141923.259
 436.3761921.355 451.6221920.827  473.881917.225 479.6741916.076 489.6661916.074
  493.461917.277 502.6481921.629  509.651922.199 602.9081921.357 669.5221921.984
 811.4711920.342 950.8091922.268 992.6111925.2311061.2071932.0631163.296 1933.84
#Mann= 7 ,-1 , 0
       0      .1       0     310    .035       0     410      .1       0
  473.88    .045       0  493.46      .1       0     510    .035       0
 1128.55      .1       0
#XS Ineff= 2 , 0
                           510.6         1926.89
Permanent Ineff=
       F       F
Bank Sta=473.88,493.46
XS Rating Curve= 0 ,0
Exp/Cntr=0.3,0.1

Type RM Length L Ch R = 1 ,12951   ,340.9,350,355.8
XS GIS Cut Line= 4
     2092850.995      184932.264      2092931.07      185498.166
 2093007.6894885185752.7506820692093100.54129863186072.092493135
#Sta/Elev= 30
       01978.549  61.6621974.733  74.9161973.126 190.8891967.272 228.2461962.765
 293.6081957.616 359.8781951.276 386.3871947.153 409.5811942.279 459.2841933.988
 475.8511932.661 482.4781930.541 489.105 1927.15 499.0461924.407   512.31917.556
 515.6141916.887 545.4351916.907 550.4541916.236  556.741914.267 571.9571912.982
 578.8091913.198   580.31914.222 585.6621917.351 589.0881917.767 839.1951918.573
1006.6141921.3081044.198 1920.621095.4481922.5481129.615 1925.39 1169.97 1925.38
#Mann= 7 ,-1 , 0
       0      .1       0     120    .035       0     520      .1       0
  556.74    .045       0   580.3      .1       0  611.54    .035       0
  1027.4     .04       0
#XS Ineff= 2 , 0
                          618.91         1922.36
Permanent Ineff=
       F       F
Bank Sta=556.74,580.3
XS Rating Curve= 0 ,0
Exp/Cntr=0.3,0.1

Type RM Length L Ch R = 1 ,12601   ,181.6,187.4,194.1
XS GIS Cut Line= 3
     2092704.249      184920.714     2092597.352      185471.546
      2092567.42       186015.03
#Sta/Elev= 30
       0 1983.52    60.6 1982.29    90.7  1983.8   167.5 1974.64   204.3 1968.21
   237.7 1960.05   287.8 1950.44   317.9 1940.66   334.6 1939.79   351.3 1935.18
   384.5 1928.95   400.4 1926.45   452.1 1922.43   482.5 1923.92   505.1 1917.92
   541.8 1911.38   548.5 1909.28   565.2 1908.82     575 1911.21   834.3 1914.57
   857.6 1915.41   870.7 1920.31   890.5  1921.3   897.2 1924.77   906.9 1933.04
   929.9 1947.54   969.3 1974.85    1035 2016.58  1077.7 2039.95  1105.4 2050.64
#Mann= 9 ,-1 , 0
       0      .1       0      20    .035       0      30      .1       0
     330     .06       0     430      .1       0   541.8    .045       0
     575      .1       0  831.11     .04       0  931.11      .1       0
#XS Ineff= 2 , 0
                          747.85         1922.96
Permanent Ineff=
       F       F
Bank Sta=541.8,575
XS Rating Curve= 0 ,0
Exp/Cntr=0.3,0.1

Type RM Length L Ch R = 1 ,12414   ,177.1,182.7,185.2
XS GIS Cut Line= 4
2092647.48577241184906.0352495152092479.62571103185287.317388925
2092381.30767508185507.9334695892092230.23361984185865.235600231
#Sta/Elev= 30
       0  1998.3    71.1 2000.29   170.6  1990.7   242.8 1968.23   285.4 1952.54
   296.1  1946.6   306.9 1945.34   321.2 1939.79   357.9  1935.8   410.8 1932.61
   439.4 1928.95   475.5 1922.88     497 1915.02  544.841907.686   554.5 1906.38
  566.831907.686   572.4 1910.37     576 1910.53   777.4 1910.99   803.2 1912.31
   818.3 1916.85   840.3 1917.04     851 1926.13   861.7 1928.54   868.8 1936.14
   873.3 1939.52   904.4 1958.02   950.9 1980.91   993.5 1995.27  1046.1 2001.65
#Mann= 12 ,-1 , 0
       0    .035       0      50      .1       0     120    .035       0
     160     .06       0     260      .1       0     360     .06       0
  544.84    .045       0  566.83     .06       0   586.6      .1       0
   606.6    .035       0  798.13     .04       0  908.13      .1       0
#XS Ineff= 2 , 0
                          782.23         1927.28
Permanent Ineff=
       F       F
Bank Sta=544.84,566.83
XS Rating Curve= 0 ,0
Exp/Cntr(USF)=0,0
Exp/Cntr=0.5,0.3

Type RM Length L Ch R = 1 ,12231   ,45.9,46.4,46.3
XS GIS Cut Line= 2
     2092581.295      184872.435     2092001.868      185701.863
#Sta/Elev= 30
       0 1998.74      56 2004.48    75.4 2003.43   140.5 1993.55   159.5 1987.95
   207.5 1967.23   259.5 1951.02   273.7 1944.01   286.6 1943.39   305.4 1940.01
     331 1934.08   347.6 1928.61   387.9 1925.09   407.6    1919   443.6 1914.52
   515.1  1910.6  523.561906.438   535.7 1905.13  544.471906.436   557.5 1908.78
   595.7 1907.78   715.4 1909.23   823.7  1916.6   842.6 1916.77   847.3 1919.09
   863.8 1933.08   892.4 1942.32   903.9 1943.61   925.1 1941.89  1011.8 1926.75
#Mann= 11 ,-1 , 0
       0    .035       0     140     .06       0     310    .035       0
     330     .06       0  523.56    .045       0  544.47     .06       0
     570    .035       0     660     .06       0     690    .035       0
     810     .04       0     930      .1       0
#XS Ineff= 2 , 0
          514.79 1917.26  549.91         1917.26
Permanent Ineff=
       F       F
Bank Sta=523.56,544.47
XS Rating Curve= 0 ,0
Exp/Cntr=0.5,0.3

Type RM Length L Ch R = 1 ,12184   ,160.6,161.7,161.2
XS GIS Cut Line= 2
     2092541.191      184849.779     2091961.764      185679.206
#Sta/Elev= 30
       0 1999.66    50.2  2004.1    71.4 2002.47   132.7 1992.91   169.3 1981.07
   215.1 1962.27   227.1 1956.09   243.8 1952.13   255.2  1945.7     307 1937.33
   318.2 1939.34   331.2 1938.64   355.2 1932.96   371.2 1932.46   407.2 1927.56
   443.2 1913.05   511.3 1908.21  520.191906.007   527.3 1905.03  546.541906.006
   693.1 1908.19   795.4 1911.77   820.6 1916.27   843.4 1917.02   862.5 1928.21
   884.3 1932.68   899.5 1930.15   914.9 1924.59   933.7 1920.68  1011.8 1922.96
#Mann= 10 ,-1 , 0
       0    .035       0     120     .06       0     240    .035       0
     360     .06       0  520.19    .045       0  546.54     .06       0
     720    .035       0     760     .06       0     840     .04       0
     930      .1       0
#XS Ineff= 2 , 0
          516.84 1913.98  548.85         1913.85
Permanent Ineff=
       F       F
Bank Sta=520.19,546.54
XS Rating Curve= 0 ,0
Exp/Cntr=0.5,0.3

Type RM Length L Ch R = 1 ,12023   ,259.9,263.6,260
XS GIS Cut Line= 4
2092429.26769262184754.961194277 2092141.5075874185150.631338947
2092012.01554006185323.2874020762091863.33948569185625.435512552
#Sta/Elev= 30
       0 1991.93    56.6 1982.92   119.6 1969.39   141.9 1960.75   180.9 1957.22
   193.3  1958.2   242.3 1965.93   272.6 1972.27   281.3    1973   290.7 1972.02
   306.9 1968.24     322  1961.2   347.8 1946.84   392.1  1926.2   416.4 1910.43
   427.7  1906.2   481.3 1904.74   530.9 1906.15  564.031904.353   575.2 1903.22
  586.291904.352     592  1905.9   761.5 1908.78     820 1912.46   834.6 1916.55
     863 1916.27   885.3 1918.03   969.9 1930.66  1022.9 1944.94  1041.8 1951.66
#Mann= 11 ,-1 , 0
       0    .035       0     240     .06       0     380      .1       0
     480     .06       0  549.25    .035       0  564.03    .045       0
  586.29    .035       0  715.07     .07       0  725.07     .06       0
  835.07     .04       0  935.07      .1       0
#XS Ineff= 2 , 0
          446.99 1915.67  687.68         1914.13
Permanent Ineff=
       F       F
Bank Sta=564.03,586.29
XS Rating Curve= 0 ,0
Exp/Cntr(USF)=0,0
Exp/Cntr=0.3,0.1

Type RM Length L Ch R = 1 ,11759   ,371.6,370.4,369.1
XS GIS Cut Line= 3
     2092241.932      184563.194     2091978.335      185030.139
     2091714.932      185570.872
#Sta/Elev= 30
       0 2016.99    44.4 2007.67    56.9 2006.82    75.7 2008.98   149.1 2028.85
   222.7 2042.39   267.9 2053.15   285.2 2052.91   295.9 2049.21   313.1 2039.35
   339.5 2021.62   373.4 1995.78   403.5 1977.99   434.5 1955.79   452.5    1945
   482.8 1920.29  502.481901.394     509 1899.82  518.281901.396   538.1 1903.48
   681.4 1902.29   850.8 1907.99   859.6  1910.4   874.8 1918.33   903.2 1919.23
   940.5 1948.85   992.1 1972.64  1016.6 1978.34  1079.2 1981.69  1137.7 1992.83
#Mann= 9 ,-1 , 0
       0    .035       0      70      .1       0     220    .035       0
     270      .1       0  502.48    .045       0  518.28      .1       0
  666.21     .07       0  886.21     .04       0  996.21      .1       0
#XS Ineff= 2 , 0
                          676.23         1906.62
Permanent Ineff=
       F       F
Bank Sta=502.48,518.28
XS Rating Curve= 0 ,0
Exp/Cntr=0.3,0.1

Type RM Length L Ch R = 1 ,11389   ,540.1,538.4,529.7
XS GIS Cut Line= 2
     2091827.891      184500.228     2091330.929      185524.534
#Sta/Elev= 30
       0 2024.83    63.1 2015.91   121.4 2004.46   179.8 2005.51     195 2002.18
   209.8 1996.12   229.4 1985.22   252.7 1968.55   267.3 1956.34   309.2 1916.19
   325.6 1903.22   340.2  1897.9   365.7 1898.75  369.031897.596     384 1896.43
  393.621897.594   551.7 1899.38   654.9 1908.13   726.7  1908.8   794.4 1912.08
   814.3 1914.61   865.3 1917.78   895.4 1921.93   948.1 1938.07   992.7 1946.05
  1015.1 1947.21  1040.3 1943.44  1075.8 1943.04  1098.4 1944.64  1138.5 1951.26
#Mann= 6 ,-1 , 0
       0      .1       0  369.03    .045       0  393.62      .1       0
     500    .035       0     720     .04       0     830      .1       0
#XS Ineff= 2 , 0
                          522.64         1909.32
Permanent Ineff=
       F       F
Bank Sta=369.03,393.62
XS Rating Curve= 0 ,0
Exp/Cntr=0.3,0.1

Type RM Length L Ch R = 1 ,10850   ,341.6,356,365.3
XS GIS Cut Line= 3
     2091225.965      184335.653     2091140.824      184899.535
     2091059.902      185439.782
#Sta/Elev= 30
       0 2026.07    74.5 2008.35   154.1 1986.76   220.5  1974.8   260.3 1963.85
   317.5 1933.58   369.8 1902.77     393 1895.09   432.9 1892.36   548.1 1894.15
  553.18 1892.86   575.5 1891.75  585.071892.861   645.2 1894.88   648.5 1895.95
   665.1 1906.81   691.6 1907.43   701.6 1914.59   708.2 1916.72   767.9 1926.89
   804.4 1929.82   874.1 1930.82   900.6 1934.71   927.2 1940.54   943.8 1941.72
   976.9  1949.3  1000.2 1952.47  1043.3 1965.79  1066.5 1966.44  1116.5 1962.37
#Mann= 5 ,-1 , 0
       0      .1       0  553.18    .045       0  585.07      .1       0
  680.27     .04       0  820.27      .1       0
#XS Ineff= 2 , 0
          426.36 1906.84
Permanent Ineff=
       F       F
Bank Sta=553.18,585.07
XS Rating Curve= 0 ,0
Exp/Cntr=0.3,0.1

Type RM Length L Ch R = 1 ,10494   ,343.4,349.8,348.4
XS GIS Cut Line= 3
      2091135.64      184299.403     2090838.685      184771.359
     2090489.206      185192.051
#Sta/Elev= 30
       0 1987.24    71.7 1957.72   120.5 1943.18     157 1934.81     250 1922.79
   331.4 1906.79   370.3 1892.72   429.8 1889.51     533 1890.17  547.331888.455
   555.9 1887.16  570.041888.454   581.6 1891.18   595.5 1899.18   618.8  1900.9
   635.1 1913.32   656.1 1923.67   688.3 1937.13   709.7  1943.3     731 1944.46
   752.3 1941.63   770.3 1935.84   795.9 1922.74   821.5 1932.91   858.8 1940.28
     924 1946.11   961.3  1944.2   969.9 1945.27  1038.1 1965.14  1104.5 1988.64
#Mann= 5 ,-1 , 0
       0      .1       0  547.33    .045       0  570.04      .1       0
  577.61     .04       0  657.61      .1       0
#XS Ineff= 2 , 0
          422.92 1900.13
Permanent Ineff=
       F       F
Bank Sta=547.33,570.04
XS Rating Curve= 0 ,0
Exp/Cntr=0.3,0.1

Type RM Length L Ch R = 1 ,10145   ,354.4,351.1,354.7
XS GIS Cut Line= 3
     2090980.959      184177.646      2090575.63      184556.672
     2090227.024      184974.924
#Sta/Elev= 30
       0  1940.6    55.8 1945.25   103.3 1960.27   163.9 1984.09   197.6 1991.96
   210.3 1992.31   226.6 1989.49   247.5 1982.51   291.2 1962.43   353.6 1930.72
   404.2 1891.83   411.3 1888.11   512.1 1888.19   537.6 1887.11  547.081884.594
   558.5 1883.04  568.181884.592   581.8 1888.53   593.8 1895.27   619.1 1895.89
   632.2 1907.62   674.9 1929.36   731.4 1951.54   756.5 1956.21   791.5 1958.27
     866 1968.62   931.2 1981.39  1008.2    1991  1072.1 2004.84  1099.4 2008.46
#Mann= 4 ,-1 , 0
       0      .1       0  547.08    .045       0  568.18     .04       0
  774.93      .1       0
#XS Ineff= 2 , 0
          436.68 1899.47
Permanent Ineff=
       F       F
Bank Sta=547.08,568.18
XS Rating Curve= 0 ,0
Exp/Cntr=0.3,0.1

Type RM Length L Ch R = 1 ,9794    ,348.1,350,345.4
XS GIS Cut Line= 3
     2090719.912      183827.361     2090398.651      184264.288
     2089958.873      184623.063
#Sta/Elev= 30
       0 2114.79    62.9 2099.72   114.5  2081.7   229.5 2037.47   297.6 2020.51
   323.6 2011.75   372.7 1987.29   404.7 1967.44   429.2 1954.35   449.5 1940.96
   467.6 1932.71   480.6 1919.44   510.6 1898.12   526.9 1883.11  530.13 1881.43
     544 1880.15  551.461881.432   562.6 1884.85   641.9 1883.26   699.1 1886.04
   714.7 1894.05   739.9 1895.47   747.7 1903.57   753.8 1907.91   793.5 1926.85
   830.8 1941.39   938.2 1959.91  1001.7 1964.52  1052.5 1962.99  1109.9 1966.19
#Mann= 6 ,-1 , 0
       0      .1       0  530.13    .045       0  551.46      .1       0
  692.32     .04       0  752.32    .035       0  842.32      .1       0
#XS Ineff= 2 , 0
                          668.77         1904.97
Permanent Ineff=
       F       F
Bank Sta=530.13,551.46
XS Rating Curve= 0 ,0
Exp/Cntr=0.3,0.1

Type RM Length L Ch R = 1 ,9444    ,349.6,350,354
XS GIS Cut Line= 3
     2090508.559      183595.426     2090163.104      184013.566
     2089790.254      184440.049
#Sta/Elev= 30
       0 2032.17    38.6 2004.18    51.5 1996.09    67.8 1988.39    82.4 1979.77
    98.2 1973.22   190.6 1943.59   247.2 1933.83     311    1926   359.1 1924.56
     394 1921.87   434.4 1915.44   491.9 1901.54     510 1893.29   532.41878.612
   536.2 1877.33   549.5 1877.28  557.931878.612   565.9  1880.2   701.3 1881.09
   745.5 1886.47   767.4 1892.28   789.6 1892.05   805.1  1896.5   837.1 1900.09
   880.7 1901.37   936.1  1906.3   959.4 1909.67  1015.8  1921.7  1108.9 1951.16
#Mann= 7 ,-1 , 0
       0      .1       0   532.4    .045       0  557.93      .1       0
  612.38    .035       0  732.38     .04       0  872.38      .1       0
 1032.38    .035       0
#XS Ineff= 2 , 0
                          667.05         1892.98
Permanent Ineff=
       F       F
Bank Sta=532.4,557.93
XS Rating Curve= 0 ,0
Exp/Cntr=0.3,0.1

Type RM Length L Ch R = 1 ,9094    ,520.6,525.2,525.2
XS GIS Cut Line= 3
     2090237.309      183421.522     2089862.269      183843.546
     2089428.093      184169.178
#Sta/Elev= 30
       0 1999.06    22.3 1990.33      73 2005.58   105.7 2010.44   123.3 2011.24
   156.7 2005.97   242.6 1984.69   268.2 1987.12   298.4 1986.34   321.7 1983.09
   335.6  1982.9   360.3 1973.79   386.6 1960.87   426.2    1935   510.3 1891.88
   544.9 1876.24  556.45 1875.23   568.7 1873.99  578.16 1875.23   585.1 1878.13
   640.7 1875.98   750.8 1879.28     786 1882.25   809.4 1889.05   839.9 1889.62
   851.7 1895.53   993.6 1938.65  1037.3 1940.64  1085.5 1936.83  1107.3 1937.11
#Mann= 6 ,-1 , 0
       0      .1       0  556.45    .045       0  578.16      .1       0
  584.59    .035       0  764.59     .04       0  924.59    .035       0
Bank Sta=556.45,578.16
XS Rating Curve= 0 ,0
Exp/Cntr=0.3,0.1

Type RM Length L Ch R = 1 ,8568    ,117.1,115.6,112.7
XS GIS Cut Line= 2
     2089944.211      183141.721     2089041.433      183788.423
#Sta/Elev= 30
       0 1913.32    24.6 1920.14    40.3 1922.63    71.4 1925.88    88.7 1925.91
   213.9 1905.76   254.2 1908.92   278.1 1916.54   318.3 1923.15   351.4 1925.25
   381.8 1920.83   414.7 1902.66     457 1872.89   464.1 1871.21  485.461870.788
     497 1869.16  509.481870.788   513.4 1872.17     569 1871.98   661.8 1877.91
   700.7 1878.08   779.5 1881.89   840.3  1887.5   859.6 1891.98   883.8  1892.4
   896.7  1900.4   988.7 1935.51  1078.1 1961.43    1095 1964.81  1110.5 1965.07
#Mann= 10 ,-1 , 0
       0     .06       0      60      .1       0     130     .08       0
     230      .1       0  485.46    .045       0  509.48     .07       0
     730    .035       0     740     .06       0     900     .04       0
     970      .1       0
Bank Sta=485.46,509.48
XS Rating Curve= 0 ,0
Exp/Cntr=0.3,0.1
